HEC-RAS study Blanche_Brook.prj: Stephenville Model

--- Blanche_Brook.g01 (geometry) --- (continued)

Type RM Length L Ch R = 1 ,2194.843,20.394,20.418,20.397
Node Photo=\HecRas Photos\BB19.JPG
BEGIN DESCRIPTION:
2008 Survey Section
END DESCRIPTION:
Node Name=BB19
XS GIS Cut Line= 4
299791.2326369925379291.28981196 299517.90990038 5379272.0366088
299447.815151001  5379267.099045  299447.66412915379267.08840682
#Sta/Elev= 13
-219.391      12  54.609    11.9  63.569   11.21  78.309    11.7  85.689    8.37
  87.549    7.72  90.509    7.91  95.409    8.28 105.879    8.39 110.479   10.92
 118.569   11.22 121.099   12.43 125.029   12.45
#Mann= 3 , 0 , 0
-219.391     .06       0  78.309    .033       0 118.569     .06       0
Levee=-1,78.33,11.7,0,,,Levee 9,
Bank Sta=78.309,118.569
XS Rating Curve= 0 ,0
Exp/Cntr=0.3,0.1

Type RM Length L Ch R = 1 ,2174.425,20.399,20.873,21.196
BEGIN DESCRIPTION:
Interpolated Section
END DESCRIPTION:
Node Name=BB18a
XS GIS Cut Line= 2
299504.4966704925379251.04732196299448.2787261735379246.45810201
#Sta/Elev= 16
  31.575  12.533  37.256   11.98  38.764  11.479   45.33    9.75  50.589    9.76
   56.51   7.963  58.002   7.606   60.37   7.717  64.289   7.928  68.497   7.982
  72.663   8.974  76.342  11.105  79.515  11.914  82.813  12.121  84.837  12.811
   87.98  12.945
#Mann= 3 , 0 , 0
  31.575     .06       0  37.256    .033       0  79.515     .06       0
Bank Sta=37.256,79.515
XS Rating Curve= 0 ,0
Exp/Cntr=0.3,0.1

Type RM Length L Ch R = 1 ,2153.552,17.891,18.471,17.928
Node Photo=\HecRas Photos\BB18).JPG
BEGIN DESCRIPTION:
2008 Survey Section
END DESCRIPTION:
Node Name=BB18
XS GIS Cut Line= 2
299492.3074642465379231.14339987299450.9894636985379223.16975064
#Sta/Elev= 7
  34.266   13.18  38.516   12.62  44.556    7.98  54.036    7.49  61.846    7.62
  70.046   12.78  76.346   13.45
#Mann= 3 , 0 , 0
  34.266     .06       0  38.516    .033       0  70.046     .06       0
#XS Ineff= 2 , 0
       0      40   13.18      68       0   13.18
Permanent Ineff=
       F       F
Bank Sta=38.516,70.046
XS Rating Curve= 0 ,0
Exp/Cntr=0.5,0.3

Type RM Length L Ch R = 3 ,2151.76 ,,,
Node Photo=\HecRas Photos\Main St Bridge.JPG
BEGIN DESCRIPTION:
Main Street Bridge
END DESCRIPTION:
Bridge Culvert--1,0,-1,-1, 0
Deck Dist Width WeirC Skew NumUp NumDn MinLoCord MaxHiCord MaxSubmerge Is_Ogee
1.79,16.52,1.6,0, 6, 6, , , 0.98, 0, 1,1,,
      34      42      42    66.4    66.4   73.77
   13.18   13.64   13.64   13.64   13.64   13.18
       0       0   11.86   11.86       0       0
      34      55      55    79.4    79.4      90
   13.64   13.64   13.64   13.64   13.64   13.18
       0       0   11.86   11.86       0       0
BR Coef=-1 , 0 , 0 ,, 0 ,,,0.8,-1,,0,
WSPro=,,,, 1 ,,,, 0 ,,,, 0 ,,,,-1 ,-1 ,-1 , 0 , 0 , 0 , 0 , 0
BC Design=,, 0 ,, 0 ,,,,,,
BC Use User HTab Curves=0
BC User HTab FreeFlow(D)= 0

Type RM Length L Ch R = 1 ,2135.081,15.08,16.997,18.315
Node Photo=\HecRas Photos\BB17.JPG
BEGIN DESCRIPTION:
2008 Survey Section
END DESCRIPTION:
Node Name=BB17
XS GIS Cut Line= 3
299496.4254602915379214.64401857 299423.53082417 5379198.9436354
299423.4056953135379198.91668457
#Sta/Elev= 9
  46.502   13.46  50.252   13.04  54.942   10.68  58.752     7.8  65.752    7.35
  71.992    6.63  76.042    7.21  85.552   13.23  87.442   13.42
#Mann= 3 , 0 , 0
  46.502     .06       0  50.252    .046       0  85.552     .06       0
#XS Ineff= 2 , 0
       0      55   13.46    79.4       0   13.33
Permanent Ineff=
       F       F
Bank Sta=50.252,85.552
XS Rating Curve= 0 ,0
Exp/Cntr=0.5,0.3

Type RM Length L Ch R = 1 ,2118.084,13.884,14.611,14.929
BEGIN DESCRIPTION:
Interpolated Section
END DESCRIPTION:
Node Name=BB16a
XS GIS Cut Line= 2
299534.9270052745379217.40501632299436.0913379175379177.61947227
#Sta/Elev= 19
  21.564  11.589  29.898  11.337  34.077  10.871  40.321  10.197  48.789   8.838
  54.427   8.744  58.529   9.037  64.346   8.812  69.824   8.543   73.08    7.04
   78.24     6.9   83.68    7.06  87.465   8.581   87.67   8.693  91.663   9.256
   94.27   9.041 104.767  10.544 109.188  11.361 113.505  11.694
#Mann= 3 , 0 , 0
  21.564     .06       0  58.529    .046       0  91.663     .06       0
Levee=-1,58.5,9.04,-1,91.63,9.26,Levee 10,Levee 11
Bank Sta=58.529,91.663
XS Rating Curve= 0 ,0
Exp/Cntr=0.3,0.1

Type RM Length L Ch R = 1 ,2103.473,62.135,67.06,69.219
Node Photo=\HecRas Photos\BB16.JPG
BEGIN DESCRIPTION:
2008 Survey Section
END DESCRIPTION:
Node Name=BB16
XS GIS Cut Line= 3
299560.8505432135379219.22100146299431.1658399995379155.81049989
299171.2704446495379028.73230974
#Sta/Elev= 14
   9.798  9.9811  28.225  9.8193  58.194  9.6958  64.235 10.3417  80.869   9.812
  85.381  7.0383  93.224  6.9383  101.83  7.0648 107.248  9.9192  113.17 10.0143
 117.036  8.9934 132.605  9.2891 145.565 10.2111 434.865      12
#Mann= 3 , 0 , 0
   9.798     .06       0  80.869    .033       0 107.248     .06       0
Levee=-1,64.06,10.34,-1,113.2,10.02,Levee 10,Levee 11
Bank Sta=80.869,107.248
XS Rating Curve= 0 ,0
Exp/Cntr=0.3,0.1

Type RM Length L Ch R = 1 ,2036.414,63.11,73.01,76.529
BEGIN DESCRIPTION:
Interpolated Section
END DESCRIPTION:
Node Name=BB15a
XS GIS Cut Line= 3
299576.286576624 5379193.2462929299457.8118981535379056.50459352
 299446.734296345379043.71899143
#Sta/Elev= 25
  18.288  10.086  35.306   9.961  36.247   9.956  56.514   9.737  62.983   9.215
  64.098   9.195  68.562   9.497  74.144   9.436  83.277   9.205  83.924   9.049
  87.245   7.156  88.091   6.869  89.432   6.871  93.411    6.69  95.334   6.379
 101.878   6.549 105.997   8.102 107.072   8.131   110.5   8.133 113.439   7.569
 120.637   7.587 121.444   7.904 125.277   8.682 128.326   9.409 135.131   9.641
#Mann= 3 , 0 , 0
  18.288     .06       0  83.277    .033       0 128.326     .06       0
Levee=-1,68.46,9.51,-1,110.58,8.14,Levee 10,Levee 11
Bank Sta=83.277,128.326
XS Rating Curve= 0 ,0
Exp/Cntr=0.3,0.1

Type RM Length L Ch R = 1 ,1963.404,73.311,66.886,63.087
Node Photo=\HecRas Photos\BB15.JPG
BEGIN DESCRIPTION:
2008 Survey Section
END DESCRIPTION:
Node Name=BB15
XS GIS Cut Line= 2
299607.3590964275379171.46521768 299574.641529385379050.81918919
#Sta/Elev= 15
  35.074    10.2  51.414   10.11  69.854    9.75  76.754    8.51  85.894    8.66
  94.204    8.52  97.814    6.67  99.804    6.71 103.424    6.39 105.174    5.77
 112.884    6.16 121.794    5.86 122.324     6.5 126.844    9.23 131.314    9.02
#Mann= 3 , 0 , 0
  35.074     .06       0  94.204    .042       0 126.844     .06       0
Levee=-1,85.97,8.66,-1,126.85,9.23,Levee 10,Levee 11
Bank Sta=94.204,126.844
XS Rating Curve= 0 ,0
Exp/Cntr=0.3,0.1

Type RM Length L Ch R = 1 ,1896.518,77.456,67.155,64.169
BEGIN DESCRIPTION:
Interpolated Section
END DESCRIPTION:
Node Name=BB14a
XS GIS Cut Line= 3
299737.3291123175379261.62883142299683.0450958425379150.14230296
299615.5339537075379011.49038739
#Sta/Elev= 26
 -28.087      10  95.913   9.077 116.225   8.979 128.421   8.851  134.74   8.812
 139.148   8.737 147.726   8.039 148.666   8.037 159.088   8.031 165.986   7.934
 169.418   8.034 171.695   7.646 173.906   6.632 174.604   6.461 176.379   6.389
 176.443   6.383 178.357   6.036 180.879   5.817 183.055   5.396  189.89   5.787
 195.446    5.84  197.79   6.453  198.26   6.906 199.553    7.71 202.267   8.622
  206.23   8.496
#Mann= 3 , 0 , 0
 -28.087     .06       0 169.418    .042       0 202.267     .06       0
Levee=-1,169.43,8.04,-1,202.25,8.62,Levee 10,Levee 11
Bank Sta=169.418,202.267
XS Rating Curve= 0 ,0
Exp/Cntr=0.3,0.1

Type RM Length L Ch R = 1 ,1829.363,25.942,26.793,25.989
Node Photo=\HecRas Photos\BB14.JPG
BEGIN DESCRIPTION:
2008 Survey Section
END DESCRIPTION:
Node Name=BB14
XS GIS Cut Line= 4
 300018.941218095379405.12798696299775.1360805385379123.25360864
299683.6317775725379017.46125836299512.3234784755378819.40382285
#Sta/Elev= 17
    -334      10     -12       8  38.685    7.95  77.575    7.78  85.135     7.8
 101.795    7.55 122.515     7.3 129.345    7.71 132.825    6.24 135.025    6.06
 137.315     5.5 142.935    5.02 153.735    5.73 157.315    8.04 163.135    7.97
     299       6     425       8
#Mann= 3 , 0 , 0
    -334     .06       0 129.345    .033       0 157.315     .06       0
Levee=-1,129.53,7.71,0,,,Levee 10,
Bank Sta=129.345,157.315
XS Rating Curve= 0 ,0
Exp/Cntr=0.3,0.1

Type RM Length L Ch R = 1 ,1802.569,18.545,19.397,20.067
BEGIN DESCRIPTION:
Interpolated Section
END DESCRIPTION:
Node Name=BB13a
XS GIS Cut Line= 3
299770.3005188575379077.14364587 299647.980331885378938.98585892
299477.9950323325378746.99144345
#Sta/Elev= 26
   39.21   9.609   65.75   9.153  70.909   9.086  74.035   9.012  82.278   8.278
  88.273   7.755  94.125   6.267  95.724   5.954  96.418    5.94 101.079   6.051
 103.454   5.402 104.956   5.307 106.518   5.051 110.354     4.8 112.758   5.119
 113.772   5.587 114.228   5.452 116.905    6.98 121.603   7.444 127.017   7.659
 139.676   6.414 140.944   6.415 151.084   7.299 167.569   7.129     260       6
     424       8
#Mann= 3 , 0 , 0
   39.21     .06       0  74.035    .033       0 127.017     .06       0
Levee=0,,,-1,127.25,7.67,,Levee 12
Bank Sta=74.035,127.017
XS Rating Curve= 0 ,0
Exp/Cntr=0.3,0.1

Type RM Length L Ch R = 1 ,1783.172,15.654,15.552,15.894
Node Photo=\HecRas Photos\BB13.JPG
BEGIN DESCRIPTION:
2008 Survey Section
END DESCRIPTION:
Node Name=BB13
XS GIS Cut Line= 3
299767.7410278315379048.98009851299675.7161904865378932.64681357
299621.7735092465378864.45512219
#Sta/Elev= 14
    7.22   10.81   30.31    9.94   39.75    7.98   43.63    5.49   44.69    4.97
   54.39    4.64   57.92    5.15   59.41    5.94   60.08     5.7   64.01    8.29
   70.91    9.01   78.86    9.29   97.45    6.93  138.41    6.52
#Mann= 3 , 0 , 0
    7.22     .06       0   30.31    .033       0   78.86     .06       0
Levee=0,,,-1,78.94,9.29,,Levee 12
#XS Ineff= 2 , 0
       0      37   10.63      70       0    9.29
Permanent Ineff=
       F       F
Bank Sta=30.31,78.86
XS Rating Curve= 0 ,0
Exp/Cntr=0.5,0.3

Type RM Length L Ch R = 3 ,1780.69 ,,,
Node Photo=\HecRas Photos\Minnesota Bridge.JPG
BEGIN DESCRIPTION:
Minnesota Drive Bridge
END DESCRIPTION:
Bridge Culvert--1,0,-1,-1, 0
Deck Dist Width WeirC Skew NumUp NumDn MinLoCord MaxHiCord MaxSubmerge Is_Ogee
2.48,11.33,1.6,0, 6, 6, , , 0.98, 0, 1,1,,
      10      40      40    66.7    66.7   78.86
    10.6      11      11      11      11    9.29
       0       0    9.23    9.23       0       0
      10      30      30    56.7    56.7      78
    9.54      11      11      11      11    9.02
       0       0    9.23    9.23       0       0
BR Coef=-1 , 0 , 0 ,, 0 ,,,0.8,-1,,0,
WSPro=,,,, 1 ,,,, 0 ,,,, 0 ,,,,-1 ,-1 ,-1 , 0 , 0 , 0 , 0 , 0
BC Design=,, 0 ,, 0 ,,,,,,
BC Use User HTab Curves=0
BC User HTab FreeFlow(D)= 0

Type RM Length L Ch R = 1 ,1767.620,17.554,40.58,15.484
Node Photo=\HecRas Photos\BB12.JPG
BEGIN DESCRIPTION:
2008 Survey Section
END DESCRIPTION:
Node Name=BB12
XS GIS Cut Line= 4
  299780.36883335379040.20944591   299780.192571  5379039.984218
299702.147574001  5378940.258348299702.0489681715378940.13234951
#Sta/Elev= 12
   -.286     9.5  22.184    9.58  30.134    7.27  34.894    5.65  36.384    5.05
  49.834    4.59  52.314    5.03  53.194    5.12  56.444    5.97  64.794     9.5
  94.384    8.39 126.794    8.15
#Mann= 3 , 0 , 0
   -.286     .06       0  22.184    .045       0  64.794     .06       0
Levee=-1,22.32,9.58,-1,64.93,9.5,Levee 13,Levee 12
#XS Ineff= 2 , 0
       0      29    9.58      58       0     9.5
Permanent Ineff=
       F       F
Bank Sta=22.184,64.794
XS Rating Curve= 0 ,0
Exp/Cntr=0.5,0.3

River Reach=Warm Creek      ,DS of Noels Pond
Reach XY= 30
 301308.01421022 5380143.6762537 301242.805165565380121.99231218
301198.4108947565380127.94205981301172.3235397485380106.88910664
301216.2601376575380030.00006031301202.9876237055379952.19566818
301250.1279318785379808.94405208 301240.974473985379778.73764102
301161.3393902715379741.20846364301102.2995868335379650.58923046
301011.2226807525379665.23476309300932.0452699395379642.35111835
300886.2779804535379668.89614625300855.613896496 5379628.6209315
 300821.288429385379619.00980071300753.0951680455379711.45972547
300686.2749253935379755.39632338300518.3089729735379731.59733285
300498.1713655985379720.61318337300469.7956461175379650.13155756
 300440.046907955379650.13155756300389.7028895135379747.61588417
300380.5494316185379850.13461262300333.4091234455379857.91505183
 300227.686684735379818.09750998300091.3001620565379696.35651995
300060.1784052035379443.72108197 299964.067097285379178.72847584
299881.2283033095379131.13049478299764.8049859475379000.93201073
Reach Upstream Storage Area=Noel's Pond

Type RM Length L Ch R = 1 ,2889.005,22.271,16.555,15.405
Node Photo=\HecRas Photos\W23.JPG
BEGIN DESCRIPTION:
2008 Survey Section
END DESCRIPTION:
Node Name=W23
XS GIS Cut Line= 3
301359.3742884185379993.67623683301312.9991003265380088.10282464
301266.6327960865380182.51132364
#Sta/Elev= 17
  56.353      26  68.953      24 161.553   23.91 185.483   23.68 197.513   23.59
 204.193    22.1 208.363   21.61 211.183   21.23  213.48   21.15  218.91   21.09
  224.13   21.17 226.743   21.34 233.183   21.76 238.473   22.18 245.763   23.46
 257.693   24.04 266.733   24.18
#Mann= 3 , 0 , 0
  56.353      .1       0 197.513     .03       0 245.763      .1       0
Bank Sta=197.513,245.763
XS Rating Curve= 0 ,0
Exp/Cntr=0.3,0.1

Type RM Length L Ch R = 5 ,2873.55 ,,,
Node Photo=\HecRas Photos\Noels Spillway.JPG
BEGIN DESCRIPTION:
Noel's Pond Outlet Weir
END DESCRIPTION:
IW Pilot Flow=0
#Inline Weir SE= 10
     195   22.75     205   22.76     205   21.95  211.05   21.95  211.05   21.15
  218.87   21.15  218.87   21.95  236.37   21.95  236.37   22.85     250   22.85
IW Dist,WD,Coef,Skew,MaxSub,Min_El,Is_Ogee,SpillHt,DesHd
15.46,0.5,1.7,0,0.98,, 0 ,,,0,1,

Type RM Length L Ch R = 1 ,2872.450,25.056,19.156,18.179
BEGIN DESCRIPTION:
Interpolated Section
END DESCRIPTION:
Node Name=W22a
XS GIS Cut Line= 3
301331.077264486 5379991.4154167301290.7424411895380089.00876538
301256.8044458955380171.12447428
#Sta/Elev= 20
  46.553      26  82.153      24 152.153  23.975 175.314   23.87 176.041  23.867
 180.439  23.807 186.957  23.332 193.423  22.088  193.59   21.39  197.83   21.15
  203.48   21.16 208.427  21.416 209.199  22.631 211.621  22.665 216.353  22.932
 218.091  23.048  220.24  23.175 225.597  23.869 234.363  24.193 241.006  24.277
#Mann= 3 , 0 , 0
  46.553      .1       0 186.957     .03       0  220.24      .1       0
#XS Ineff= 2 , 0
       0     183   23.98     216       0   24.19
Permanent Ineff=
       F       F
Bank Sta=186.957,220.24
XS Rating Curve= 0 ,0
Exp/Cntr=0.5,0.3

Type RM Length L Ch R = 3 ,2868.55 ,,,
Node Photo=\HecRas Photos\Conneticuit Bridge.JPG
BEGIN DESCRIPTION:
Noel's Pond Outlet Bridge
END DESCRIPTION:
Bridge Culvert--1,0,-1,-1, 0
Deck Dist Width WeirC Skew NumUp NumDn MinLoCord MaxHiCord MaxSubmerge Is_Ogee
5,8.25,1.6,0, 6, 6, , , 0.98, 0, 1,1,,
  152.15     188     188   210.1   210.1  234.36
   23.98    24.7    24.7    24.7    24.7   24.19
       0       0   23.92   23.92       0       0
  146.96     176     176   198.1   198.1  216.93
   24.05    24.7    24.7    24.7    24.7   24.39
       0       0   23.92   23.92       0       0
Pier Skew, UpSta & Num, DnSta & Num=  ,199.07, 2 ,187.07, 2 , 0 , 0 , 0 ,,
     .74     .74
       0   23.92
     .74     .74
       0   23.92
BR Coef=-1 , 0 , 0 ,, 0 ,,,0.8,-1,,0,
WSPro=,,,, 1 ,,,, 0 ,,,, 0 ,,,,-1 ,-1 ,-1 , 0 , 0 , 0 , 0 , 0
BC Design=,, 0 ,, 0 ,,,,,,
BC Use User HTab Curves=0
BC User HTab FreeFlow(D)= 0

Type RM Length L Ch R = 1 ,2853.295,62.32,146.599,163.025
Node Photo=\HecRas Photos\W22.JPG
BEGIN DESCRIPTION:
2008 Survey Section
END DESCRIPTION:
Node Name=W22
XS GIS Cut Line= 2
 301265.992856035380090.46296967301244.8021192545380157.14710638
#Sta/Elev= 12
 146.959   24.05 169.929   24.09 174.159      24  183.84   21.96  184.93   21.07
  188.26   21.09 193.149   21.07  197.39   21.07 197.949   21.54 198.399   24.15
 203.579   24.32 216.929   24.39
#Mann= 3 , 0 , 0
 146.959      .1       0 174.159     .03       0 198.399      .1       0
Bank Sta=174.159,198.399
XS Rating Curve= 0 ,0
Exp/Cntr=0.5,0.3

Type RM Length L Ch R = 1 ,2706.696,280.29,270.077,227.593
Node Photo=\HecRas Photos\W21.JPG
BEGIN DESCRIPTION:
2008 Survey Section
END DESCRIPTION:
Node Name=W21
XS GIS Cut Line= 2
301240.8198410325380086.71513002301170.0227037365380044.65228316
#Sta/Elev= 15
  11.439   23.74  33.699   23.39  36.529   22.35  53.519   21.96  55.749   21.07
  56.768   20.29   58.42   20.27  59.279   20.08   59.69   20.27  62.658   20.33
  63.899   20.98  67.909   22.96  78.619   23.72  86.839   26.01  93.789   26.05
#Mann= 3 , 0 , 0
  11.439      .1       0  55.749     .05       0  63.899      .1       0
Bank Sta=55.749,63.899
XS Rating Curve= 0 ,0
Exp/Cntr=0.3,0.1

Type RM Length L Ch R = 1 ,2436.619,240.8,247.162,196.133
Node Photo=\HecRas Photos\W20.JPG
BEGIN DESCRIPTION:
1:2500 Community Mapping Section
END DESCRIPTION:
Node Name=W17d
XS GIS Cut Line= 5
301285.261793047 5379792.0819097301256.3901449445379808.20191322
301181.6138240435379849.95202573301164.1513104015379859.70192918
301101.3674640025379894.75624342
#Sta/Elev= 25
       0  27.104   2.885  27.115  16.972  26.693  19.403  26.557  25.264      26
  28.865      24  33.092  21.011  34.693      20      35    19.4   36.59   19.14
   45.47   19.14   47.28   19.41   49.64   20.06  80.203  21.496  90.826  21.817
 105.025      22 140.753  23.261 144.796      24 152.108  24.937 159.534      26
 168.622      28 170.209  28.767 173.052      30 183.477  29.848 187.963      28
#Mann= 3 , 0 , 0
       0      .1       0  34.693     .05       0   49.64      .1       0
Bank Sta=34.693,49.64
XS Rating Curve= 0 ,0
Exp/Cntr=0.3,0.1

Type RM Length L Ch R = 1 ,2189.458,205.74,214.433,169.067
Node Photo=\HecRas Photos\W19.JPG
BEGIN DESCRIPTION:
1:2500 Community Mapping Section
END DESCRIPTION:
Node Name=W17c
XS GIS Cut Line= 5
301110.5621804555379618.14852348301097.8412540975379641.72226813
 301065.276012115379702.07044384301058.1526354465379715.27110689
301000.991809398 5379821.1985118
#Sta/Elev= 13
       0   25.38  21.479      24  24.096  22.803  26.172      22   29.15  20.213
  29.661      20      30    19.2      33    19.2      38   20.32 115.294  20.753
 174.782      22 207.388  22.521 230.727  23.776
#Mann= 3 , 0 , 0
       0      .1       0   29.15     .04       0      38      .1       0
Bank Sta=29.15,38
XS Rating Curve= 0 ,0
Exp/Cntr=0.3,0.1

Type RM Length L Ch R = 1 ,1975.025,192.041,193.482,126.262
Node Photo=\HecRas Photos\W18.JPG
BEGIN DESCRIPTION:
1:2500 Community Mapping Section
END DESCRIPTION:
Node Name=W17b
XS GIS Cut Line= 4
300903.6810602775379507.81192605300900.2054420385379571.91777357
300895.6535312825379655.87523864  300889.88898565379762.19908123
#Sta/Elev= 13
       0  23.107   31.56  22.204  35.677      22  50.261  20.826    64.2  20.138
  66.628      20      67    19.1      73    19.1      74      20 189.606  20.189
 199.988      22 202.569      24 254.761   25.98
#Mann= 3 , 0 , 0
       0      .1       0    64.2     .04       0 189.606      .1       0
Bank Sta=64.2,189.606
XS Rating Curve= 0 ,0
Exp/Cntr=0.3,0.1

Type RM Length L Ch R = 1 ,1781.543,78.667,89.117,103.438
BEGIN DESCRIPTION:
1:2500 Community Mapping Section
END DESCRIPTION:
Node Name=W17a
XS GIS Cut Line= 4
300724.3840894575379641.13531461300754.6662697755379681.05273412
300805.7607267865379748.40451836300825.5259704355379774.45870317
#Sta/Elev= 27
       0  22.768  19.172  22.566   27.74  22.329  28.677  22.302  39.485      22
  48.226  20.672  50.104  20.413  53.089      20      54      19      56      19
      57      20  92.195  20.082  92.433  20.107  97.114  20.616  99.501  20.872
  104.32  21.381 105.422    21.5 110.658      22 113.998  22.328 116.841  22.598
 118.488  22.754 121.125  22.992 128.626      24 151.571  25.858 153.349      26
 166.061  26.448 167.346  26.492
#Mann= 3 , 0 , 0
       0      .1       0  53.089     .04       0  92.433      .1       0
Bank Sta=53.089,92.433
XS Rating Curve= 0 ,0
Exp/Cntr=0.3,0.1

Type RM Length L Ch R = 1 ,1692.426,55.271,56.986,58.395
Node Photo=\HecRas Photos\W17.JPG
BEGIN DESCRIPTION:
2008 Survey Section
END DESCRIPTION:
Node Name=W17
XS GIS Cut Line= 2
300698.6916769585379734.14148137300700.3620475935379818.87482816
#Sta/Elev= 16
  31.486   22.57  34.656   22.48  41.026   22.32   43.79   20.55  44.706   19.93
    47.9   19.82  48.546   19.45   50.16   19.58  51.956   19.47   52.34   19.68
  54.966   19.73   57.59   19.81  60.366   19.77  63.616   20.57 111.606   21.17
 116.236   21.65
#Mann= 3 , 0 , 0
  31.486      .1       0   43.79     .05       0  63.616      .1       0
Bank Sta=43.79,63.616
XS Rating Curve= 0 ,0
Exp/Cntr=0.3,0.1

Type RM Length L Ch R = 1 ,1635.440,99.483,101.822,103.873
Node Photo=\HecRas Photos\W16.JPG
BEGIN DESCRIPTION:
2008 Survey Section
END DESCRIPTION:
Node Name=W16
XS GIS Cut Line= 3
300644.5963847925379723.98834471300643.7766037925379737.19592749
300637.9019106085379831.84376211
#Sta/Elev= 11
    17.5      24    22.8      22  30.733   20.15  36.943   19.85  40.513   19.12
  42.143   18.88  46.033   18.84   49.57   18.92  51.393   19.16  54.803   19.72
 125.563   21.33
#Mann= 3 , 0 , 0
    17.5      .1       0  36.943     .04       0  54.803      .1       0
Bank Sta=36.943,54.803
XS Rating Curve= 0 ,0
Exp/Cntr=0.3,0.1

Type RM Length L Ch R = 1 ,1533.618,162.203,157.685,116.864
BEGIN DESCRIPTION:
Interpolated Section
END DESCRIPTION:
Node Name=W15a
XS GIS Cut Line= 3
300574.4828022915379578.24269088300550.0222001485379705.20486391
300529.2801185155379812.86614477
#Sta/Elev= 18
  -90.58      22   19.42      20  38.717  18.938  48.019   18.86  53.367  18.476
  54.091  18.441  55.809   18.43  60.177  18.646  61.636  17.981  64.392  18.139
  67.481  18.427  68.841  18.633  71.199   19.27  71.632  19.353  85.705  19.559
  87.451  19.926 107.319  20.315 148.358  21.102
#Mann= 3 , 0 , 0
  -90.58      .1       0  48.019     .05       0  71.632      .1       0
Bank Sta=48.019,71.632
XS Rating Curve= 0 ,0
Exp/Cntr=0.3,0.1

Type RM Length L Ch R = 1 ,1375.933,115.399,110.024,80.619
Node Photo=\HecRas Photos\W15.JPG
BEGIN DESCRIPTION:
2008 Survey Section
END DESCRIPTION:
Node Name=W15
XS GIS Cut Line= 4
300438.6961542185379587.56423744300439.2666163955379626.41905013
300439.5602225855379646.41689395300441.2129295155379758.98459923
#Sta/Elev= 19
     -31      24     -29      22     -27      20     -22      18   -1.41   17.37
   7.859   17.06   17.61   17.33  31.149    17.5   40.32   18.34  40.369   18.33
  42.579   16.65  45.689   16.82   47.32   17.21  50.709    17.5  53.859   18.77
  69.739   18.84  71.709   19.72  94.129   20.07 140.439   20.75
#Mann= 3 , 0 , 0
     -31      .1       0   40.32    .045       0  53.859      .1       0
Bank Sta=40.32,53.859
XS Rating Curve= 0 ,0
Exp/Cntr=0.3,0.1

Type RM Length L Ch R = 1 ,1265.909,88.883,82.766,73.503
BEGIN DESCRIPTION:
Interpolated Section
END DESCRIPTION:
Node Name=W14a
XS GIS Cut Line= 3
300370.6541418085379721.89731956300384.7266877325379740.56782603
300435.0195849435379807.29305599
#Sta/Elev= 21
    11.9      22   18.49      20   30.14      18   35.28  17.705  46.005  17.259
  48.973  16.967  51.589  16.845  54.394  16.982   55.05   16.66   57.68   16.43
   59.67    16.5  61.031  16.606  62.371  16.776  64.352  17.391  65.938  17.451
  74.342  17.963  74.403  17.986  75.581    18.6   83.57  20.416  89.684  20.476
 118.816  20.744
#Mann= 3 , 0 , 0
    11.9      .1       0  54.394    .045       0  64.352      .1       0
Levee=-1,54.46,16.97,0,,,Levee 21,
Bank Sta=54.394,64.352
XS Rating Curve= 0 ,0
Exp/Cntr=0.3,0.1

Type RM Length L Ch R = 1 ,1183.143,20.173,34.556,39.04
Node Photo=\HecRas Photos\W14.JPG
BEGIN DESCRIPTION:
2008 Survey Section
END DESCRIPTION:
Node Name=W14
XS GIS Cut Line= 3
300298.9502244315379806.31093566300374.6881692135379826.69472821
300419.7251011965379838.81577904
#Sta/Elev= 12
   -52.1      20   -23.4      18  26.333   18.19  31.403   17.15  34.043   16.05
  35.983   15.93  38.723   15.93  40.823   16.15  43.553   16.45  48.263   17.31
  53.363   20.79  72.973   20.74
#Mann= 3 , 0 , 0
   -52.1      .1       0  31.403    .045       0  48.263      .1       0
Bank Sta=31.403,48.263
XS Rating Curve= 0 ,0
Exp/Cntr=0.3,0.1

Type RM Length L Ch R = 1 ,1148.587,12.279,23.372,25.348
BEGIN DESCRIPTION:
Interpolated Section
END DESCRIPTION:
Node Name=W13a
XS GIS Cut Line= 3
300335.5427684825379796.83576298300352.6128293185379827.48588301
300385.2597630775379886.10503194
#Sta/Elev= 21
  -30.06      22  -20.03      20   -3.23      18   5.023  18.083   8.579  17.275
   14.18  17.139  16.338  16.985  18.948  15.968  19.034  15.941  22.452  15.727
  23.558  15.727  26.535  15.905  30.337  16.138  30.406  16.167  34.156  17.814
  37.084  17.983  44.315  19.428  44.687  19.429  59.571  19.753   70.01  19.894
   72.12  20.173
#Mann= 3 , 0 , 0
  -30.06      .1       0   14.18    .045       0  34.156      .1       0
Bank Sta=14.18,34.156
XS Rating Curve= 0 ,0
Exp/Cntr=0.3,0.1

Type RM Length L Ch R = 1 ,1125.215,33.473,35.913,35.28
Node Photo=\HecRas Photos\W13.JPG
BEGIN DESCRIPTION:
2008 Survey Section
END DESCRIPTION:
Node Name=W13
XS GIS Cut Line= 4
300347.5260179465379785.28417287 300347.485885715379786.86366303
300346.4538013975379827.48355279300344.3981726435379908.38722733
#Sta/Elev= 15
  -18.58      22  -11.33      20   11.07      18  23.633   18.01  28.263   16.93
  38.363   17.21  41.873   15.87  46.323   15.59  54.453   15.93   56.92   17.21
  59.033   18.41  71.663   18.51  89.513   19.07 102.033   19.32 104.563   19.79
#Mann= 3 , 0 , 0
  -18.58      .1       0  38.363    .045       0   56.92      .1       0
Levee=-1,38.24,17.21,0,,,Levee 22,
Bank Sta=38.363,56.92
XS Rating Curve= 0 ,0
Exp/Cntr=0.3,0.1

Type RM Length L Ch R = 1 ,1089.302,36.577,37.305,37.535
BEGIN DESCRIPTION:
Interpolated Section
END DESCRIPTION:
Node Name=W12a
XS GIS Cut Line= 2
300314.0330639555379822.61789455300309.247893518 5379886.1923018
#Sta/Elev= 18
  26.012  20.791  31.138  18.404  32.844  17.815  36.524  17.602   41.33  16.638
  42.321  16.633  46.207  15.881  46.837  15.852  51.134  15.659  56.527  16.448
   56.72   16.55  59.565  17.806  67.943  18.073  76.183  18.483  79.783  18.848
  82.403  19.091  88.088  19.223  89.766  19.476
#Mann= 3 , 0 , 0
  26.012     .04       0  36.524    .045       0  59.565     .04       0
Bank Sta=36.524,59.565
XS Rating Curve= 0 ,0
Exp/Cntr=0.3,0.1

Type RM Length L Ch R = 1 ,1051.997,119.597,121.94,125.44
Node Photo=\HecRas Photos\W12.JPG
BEGIN DESCRIPTION:
2008 Survey Section
END DESCRIPTION:
Node Name=W12
XS GIS Cut Line= 2
300278.1797119045379817.14976326300273.9853621615379862.86817545
#Sta/Elev= 13
  41.591   23.68  49.111   18.69  53.161   18.16  58.451   16.07   61.74   16.07
  64.511   15.87   67.45   15.87  69.241   15.73   70.34   16.31  71.881   17.03
  81.081   18.05  84.021   19.03  87.501   19.15
#Mann= 3 , 0 , 0
  41.591     .04       0  53.161    .045       0  71.881     .04       0
Bank Sta=53.161,71.881
XS Rating Curve= 0 ,0
Exp/Cntr=0.3,0.1

Type RM Length L Ch R = 1 ,930.0570,121.399,127.112,129.974
BEGIN DESCRIPTION:
Interpolated Section
END DESCRIPTION:
Node Name=W11a
XS GIS Cut Line= 2
300189.3136271425379758.25458379300156.4270450765379798.80645942
#Sta/Elev= 18
  39.315  21.413  46.614  16.596  47.782  16.152  50.545   15.79  54.876  14.621
  55.679  14.453   60.62   14.41    63.1   14.36   66.08   14.41  68.443  14.617
  69.449  14.906  69.821  15.086  72.699  16.075  75.663  16.068  82.605  16.545
  86.691   17.16  87.216  17.181  91.526  17.564
#Mann= 3 , 0 , 0
  39.315     .04       0  50.545    .045       0  72.699     .04       0
Bank Sta=50.545,72.699
XS Rating Curve= 0 ,0
Exp/Cntr=0.3,0.1

Type RM Length L Ch R = 1 ,802.9447,71.609,75.267,71.522
Node Photo=\HecRas Photos\W11.JPG
BEGIN DESCRIPTION:
2008 Survey Section
END DESCRIPTION:
Node Name=W11
XS GIS Cut Line= 2
 300109.024391465379677.44797171300053.624571032 5379697.0932981
#Sta/Elev= 14
  52.439   19.05  60.639   13.67  67.509   12.77   70.92    12.8  74.999   12.75
   77.01   12.66  78.429   12.53   79.67   12.67  81.389   12.61  82.689   12.83
  86.889   14.84  90.719   14.58 105.649   15.24 111.219   15.91
#Mann= 3 , 0 , 0
  52.439     .04       0  60.639    .045       0  82.689     .04       0
Levee=0,,,-1,86.82,14.83,,Levee 23
Bank Sta=60.639,82.689
XS Rating Curve= 0 ,0
Exp/Cntr=0.3,0.1

Type RM Length L Ch R = 1 ,727.6773,79.11,78.888,80.462
BEGIN DESCRIPTION:
Interpolated Section
END DESCRIPTION:
Node Name=W10a
XS GIS Cut Line= 2
300099.889136565 5379608.0488858300038.2185467355379634.14028919
#Sta/Elev= 20
  50.773   18.02   57.42  15.077  58.467   14.96  62.989   13.48  69.061  11.985
  70.106  11.687   71.81   11.63   73.84    11.6   75.81   11.64  77.044  11.675
  77.804  11.749  81.308  12.491  83.682  13.531  86.819  14.279  89.043  13.666
  91.899  12.995  97.556  13.624  109.94  13.945 114.019  14.165 117.736  14.562
#Mann= 3 , 0 , 0
  50.773     .04       0  62.989    .045       0  83.682     .04       0
Levee=0,,,-1,86.88,14.29,,Levee 23
Bank Sta=62.989,83.682
XS Rating Curve= 0 ,0
Exp/Cntr=0.3,0.1

Type RM Length L Ch R = 1 ,648.7893,69.05,68.73,68.507
Node Photo=\HecRas Photos\W10.JPG
BEGIN DESCRIPTION:
2008 Survey Section
END DESCRIPTION:
Node Name=W10
XS GIS Cut Line= 2
300092.3868587025379526.86943979300002.014689702   5379565.73747
#Sta/Elev= 18
  44.297   16.94  50.107   16.49   56.85      12  58.897   10.66   59.71   10.53
  60.207   10.33   61.09    10.5  62.927   10.43   64.42    10.6  66.967   10.56
   68.04   10.78  72.507   10.88   74.47   11.73  79.667   13.85  86.267   11.24
  93.617   12.34 115.007   12.67 119.837   13.15
#Mann= 3 , 0 , 0
  44.297     .04       0   56.85    .045       0   74.47     .04       0
Levee=0,,,-1,79.82,13.84,,Levee 23
Bank Sta=56.85,74.47
XS Rating Curve= 0 ,0
Exp/Cntr=0.3,0.1

Type RM Length L Ch R = 1 ,580.0592,74.519,73.956,72.988
BEGIN DESCRIPTION:
Interpolated Section
END DESCRIPTION:
Node Name=W9a
XS GIS Cut Line= 2
300073.6423346195379462.06826613299999.8798686985379497.88561736
#Sta/Elev= 27
  49.643   14.19  54.069  13.688  55.739  13.612  61.845  11.566  63.644  10.018
   64.55    9.82  64.963   9.522  66.338   9.285   67.81    9.35  69.317   9.354
  69.594    9.36   70.43    9.51  72.035   9.585   72.61    9.82  73.741    9.96
  77.476  10.826  79.808  10.866   87.65  12.327  91.386   11.59  94.878  11.015
  98.263   11.33 102.927  11.637 107.819  11.648 111.971   11.38 114.559  11.722
 126.353  11.921 131.642   12.22
#Mann= 3 , 0 , 0
  49.643     .04       0  61.845    .045       0  79.808     .04       0
Levee=0,,,-1,87.75,12.34,,Levee 23
Bank Sta=61.845,79.808
XS Rating Curve= 0 ,0
Exp/Cntr=0.3,0.1

Type RM Length L Ch R = 1 ,506.1030,11.553,11.974,12.929
Node Photo=\HecRas Photos\W09.JPG
BEGIN DESCRIPTION:
2008 Survey Section
END DESCRIPTION:
Node Name=W9
XS GIS Cut Line= 4
300068.2414353455379380.97935433300056.1398469045379388.59785433
299980.8645969775379435.98704577299968.0013722145379444.08503045
#Sta/Elev= 18
   3.305      12  17.605   11.23  22.255   10.54  30.425   10.42  32.315    8.43
    33.7    8.34  35.145    8.16  38.705     8.2      40    8.48  41.375    8.59
  47.325    10.9  62.535   10.61  70.055   10.93  80.505   10.83  85.045   10.21
  87.875   10.88 106.555   11.22 121.755      12
#Mann= 3 , 0 , 0
   3.305     .04       0  30.425    .045       0  47.325     .04       0
Levee=0,,,-1,47.37,10.91,,Levee 23
Bank Sta=30.425,47.325
XS Rating Curve= 0 ,0
Exp/Cntr=0.3,0.1

Type RM Length L Ch R = 1 ,494.1285,15.27,14.846,14.427
Node Photo=\HecRas Photos\W08.JPG
BEGIN DESCRIPTION:
2008 Survey Section
END DESCRIPTION:
Node Name=W8
XS GIS Cut Line= 4
300090.8916212315379368.46471498300058.5959418035379379.98234975
299964.7175778395379413.46226807299937.0287000835379423.33697537
#Sta/Elev= 19
       0  12.547  14.348  12.252  21.386      12  26.323  11.318  34.288   11.05
  43.138   10.47  55.978   10.64  57.898     9.9  58.348    7.99  67.408    8.16
  67.688    9.87  69.908   10.63  82.668   10.75  98.548   10.55 110.268   10.82
 133.958   11.74  158.33      12 162.957      14 163.355  14.007
#Mann= 3 , 0 , 0
       0     .04       0  55.978    .033       0  69.908     .04       0
Levee=-1,56.09,10.64,0,,,Levee 24,
#XS Ineff= 2 , 0
       0      58   10.64               0
Permanent Ineff=
       F       F
Bank Sta=55.978,69.908
XS Rating Curve= 0 ,0
Exp/Cntr=0.5,0.3

Type RM Length L Ch R = 3 ,493.61  ,,,
Node Photo=\HecRas Photos\Miss Bridge.JPG
BEGIN DESCRIPTION:
Miss Drive Bridge
END DESCRIPTION:
Bridge Culvert--1,0,-1,-1, 0
Deck Dist Width WeirC Skew NumUp NumDn MinLoCord MaxHiCord MaxSubmerge Is_Ogee
0.52,12.87,1.6,0, 6, 6, , , 0.98, 0, 1,1,,
   55.98    58.4    58.4    67.6    67.6   69.91
   10.64   10.65   10.65   10.65   10.65   10.63
       0       0    9.86    9.86       0       0
   31.34    41.1    41.1    50.3    50.3   57.72
   10.63   10.65   10.65   10.65   10.65   10.63
       0       0    9.86    9.86       0       0
BR Coef=-1 , 0 , 0 ,, 0 ,,,0.8,-1,,0,
WSPro=,,,, 1 ,,,, 0 ,,,, 0 ,,,,-1 ,-1 ,-1 , 0 , 0 , 0 , 0 , 0
BC Design=,, 0 ,, 0 ,,,,,,
BC Use User HTab Curves=0
BC User HTab FreeFlow(D)= 0

Type RM Length L Ch R = 1 ,479.2822,18.024,15.05,14.12
Node Photo=\HecRas Photos\W07.JPG
BEGIN DESCRIPTION:
2008 Survey Section
END DESCRIPTION:
Node Name=W7
XS GIS Cut Line= 3
300104.6511135465379338.87418198 300049.926581165379364.90465646
299964.7605915165379405.41502764
#Sta/Elev= 20
 -39.359      12  21.241   10.92  35.011   10.52  38.871   10.42  40.681    9.88
  40.941    8.26  43.581    7.91   45.45    7.87  46.641    7.75   48.62    7.74
  49.941    7.45   50.16    7.77  50.851    8.09  50.991    9.91  53.231   10.52
  62.391   10.75  80.321   10.49  84.271    9.94  93.421   10.73 115.551   11.48
#Mann= 3 , 0 , 0
 -39.359     .04       0  38.871    .045       0  53.231     .04       0
Levee=0,,,-1,62.47,10.76,,Levee 25
Bank Sta=38.871,53.231
XS Rating Curve= 0 ,0
Exp/Cntr=0.5,0.3

Type RM Length L Ch R = 1 ,464.2327,69.028,69.847,71.832
Node Photo=\HecRas Photos\W06.JPG
BEGIN DESCRIPTION:
2008 Survey Section
END DESCRIPTION:
Node Name=W6
XS GIS Cut Line= 2
300055.7657332375379338.69292146299958.817893427 5379403.0048548
#Sta/Elev= 17
   22.96   10.52   48.73    9.51   58.75    9.58   61.23     7.8   62.07    7.61
   64.51    7.57   65.54    7.39    68.8    7.37   70.02    7.56   72.83     7.6
   74.24    8.01      75   10.17   89.75   10.61   97.32   10.52  101.53    9.83
  114.83   10.76   139.3   11.54
#Mann= 3 , 0 , 0
   22.96     .04       0   58.75     .03       0      75     .04       0
Bank Sta=58.75,75
XS Rating Curve= 0 ,0
Exp/Cntr=0.3,0.1

Type RM Length L Ch R = 1 ,394.3861,63.972,68.222,69.71
BEGIN DESCRIPTION:
Interpolated Section
END DESCRIPTION:
Node Name=W5a
XS GIS Cut Line= 3
300115.5698633285379255.65033573300033.2517324575379284.08258489
299946.5794008885379314.01875205
#Sta/Elev= 26
     -19      10      19       8   68.09   9.179  89.294   8.613  90.275   8.614
   92.44   8.982  97.539   9.115   99.58    8.28 101.469   8.242 102.279   7.974
  102.84    7.36 104.951   7.203 106.812   7.024  109.37    7.27  110.62   8.384
 110.902   8.395 118.994   8.601 121.899   8.582 122.526   8.561 124.614   8.717
 127.687   9.281  128.75    9.36 130.906   9.161 141.076   9.734 152.738  10.105
 159.787  10.579
#Mann= 3 , 0 , 0
     -19     .04       0  97.539    .033       0 127.687     .04       0
Levee=-1,97.68,9.12,-1,128.75,9.36,Levee 26,Levee 27
Bank Sta=97.539,127.687
XS Rating Curve= 0 ,0
Exp/Cntr=0.3,0.1

Type RM Length L Ch R = 1 ,326.1642,14.443,16.892,18.313
Node Photo=\HecRas Photos\W05.JPG
BEGIN DESCRIPTION:
2008 Survey Section
END DESCRIPTION:
Node Name=W5
XS GIS Cut Line= 5
300276.8093800145379170.68468354300136.6980384355379199.28209533
300009.1614444545379225.31293948299892.9600124975379249.03022148
299881.1651905175379251.43760248
#Sta/Elev= 19
    -163      12     -20      10      34       8 110.166    7.87 127.686    7.73
 129.396    8.44 136.526    8.83 139.276    6.85 140.746     6.5 143.606    6.65
 149.266    6.75 151.736    6.57 153.196    6.91 156.066    8.46 172.866    8.99
 177.796    9.64  183.93      10 188.262  11.446 189.834      12
#Mann= 3 , 0 , 0
    -163     .04       0 136.526    .033       0 156.066     .04       0
Levee=-1,136.5,8.84,0,,,Levee 26,
Bank Sta=136.526,156.066
XS Rating Curve= 0 ,0
Exp/Cntr=0.3,0.1

Type RM Length L Ch R = 1 ,309.2723,15.642,14.996,14.953
Node Photo=\HecRas Photos\W04.JPG
BEGIN DESCRIPTION:
2008 Survey Section
END DESCRIPTION:
Node Name=W4
XS GIS Cut Line= 4
300136.303502507 5379189.7286179300007.384630526  5379210.427634
 299915.888196465379225.11816094299805.3834867285379242.86062743
#Sta/Elev= 15
      -8      10      44       8  122.57    8.66  141.46    8.73  143.48    9.36
  148.05    9.22  150.25    8.58  152.14    6.77  154.09     6.4  158.69    6.59
  165.12    6.64  169.24    8.59  176.97    9.14  202.08    9.12     314      10
#Mann= 3 , 0 , 0
      -8     .04       0  148.05    .033       0  176.97     .04       0
Levee=-1,143.55,9.35,0,,,Levee 26,
#XS Ineff= 2 , 0
       0     151    9.36     168       0    9.14
Permanent Ineff=
       F       F
Bank Sta=148.05,176.97
XS Rating Curve= 0 ,0
Exp/Cntr=0.5,0.3

Type RM Length L Ch R = 3 ,305.02  ,,,
Node Photo=\HecRas Photos\Carolina Bridge.JPG
BEGIN DESCRIPTION:
Carolina Ave Bridge
END DESCRIPTION:
Bridge Culvert--1,0,-1,-1, 0
Deck Dist Width WeirC Skew NumUp NumDn MinLoCord MaxHiCord MaxSubmerge Is_Ogee
4.25,8.94,1.6,0, 6, 6, , , 0.98, 0, 1,1,,
  143.48     155     155   163.9   163.9  176.97
    9.36    9.55    9.55    9.55    9.55    9.14
       0       0    8.55    8.55       0       0
  214.21     234     234   242.9   242.9  251.75
     9.3    9.55    9.55    9.55    9.55    9.29
       0       0    8.55    8.55       0       0
BR Coef=-1 , 0 , 0 ,, 0 ,,,0.8,-1,,0,
WSPro=,,,, 1 ,,,, 0 ,,,, 0 ,,,,-1 ,-1 ,-1 , 0 , 0 , 0 , 0 , 0
BC Design=,, 0 ,, 0 ,,,,,,
BC Use User HTab Curves=0
BC User HTab FreeFlow(D)= 0

Type RM Length L Ch R = 1 ,294.2762,85.792,40.217,25.479
Node Photo=\HecRas Photos\W03.JPG
BEGIN DESCRIPTION:
2008 Survey Section
END DESCRIPTION:
Node Name=W3
XS GIS Cut Line= 4
300134.5442039585379172.85225154300028.4277358875379191.25291856
299923.975984997 5379209.3649225299603.360395015 5379264.9598817
#Sta/Elev= 13
  95.028      10 138.628       8 202.728    9.01 214.208     9.3 228.308    9.24
 232.428    6.66 237.808    6.42 240.768    6.38 243.528     6.8 247.008       9
 251.748    9.29 287.538    8.72 612.938      10
#Mann= 3 , 0 , 0
  95.028     .04       0 228.308    .033       0 247.008     .04       0
Levee=-1,214.22,9.3,-1,251.63,9.29,Levee 26,Levee 28
#XS Ineff= 2 , 0
       0     233     9.3   243.3       0    9.29
Permanent Ineff=
       F       F
Bank Sta=228.308,247.008
XS Rating Curve= 0 ,0
Exp/Cntr=0.5,0.3

Type RM Length L Ch R = 1 ,254.0591,74.46,106.674,110.065
Node Photo=\HecRas Photos\W0.JPG
BEGIN DESCRIPTION:
2008 Survey Section
END DESCRIPTION:
Node Name=W2
XS GIS Cut Line= 6
300215.3837418395378846.99193121299986.9183204945379124.95448985
299918.8401838145379207.78178576299916.7070083875379210.37711461
299916.1888667195379211.00751191 299838.846335575379305.10633824
#Sta/Elev= 19
     -68      10      44       8      89       6     241       6 291.805    7.08
 331.375    7.29 339.445    8.51 343.725    8.55 346.775    6.59 348.565    6.16
 349.185    5.86 351.425    5.95 353.245    6.12 354.635    6.44 357.715    7.91
 365.735    7.56 380.705       8 403.195    8.85     525      10
#Mann= 3 , 0 , 0
     -68     .04       0 343.725    .033       0 357.715     .04       0
Levee=-1,343.89,8.55,-1,357.71,7.92,Levee 26,Levee 28
Bank Sta=343.725,357.715
XS Rating Curve= 0 ,0
Exp/Cntr=0.3,0.1

Type RM Length L Ch R = 1 ,147.3854,137.703,117.268,115.163
BEGIN DESCRIPTION:
Interpolated Section
END DESCRIPTION:
Node Name=W1a
XS GIS Cut Line= 3
300230.444808427 5378885.1405377299915.6107996985379079.12916934
299831.1880560285379131.14722352
#Sta/Elev= 25
-135.325      10 -46.525       8   6.675       6 234.475   7.718  249.89    8.69
 262.604   6.815 264.954   6.713  268.34    7.02  268.37    7.02 271.383   6.978
 273.551   5.906 274.823   5.655 275.264   5.488 276.833   5.554 278.107   5.659
  279.08   5.838 280.839   6.487 281.236   6.693 285.299    7.22 286.852   7.155
  292.31   7.223 297.333   7.827 303.214   8.571 310.622   9.767 313.079   9.865
#Mann= 3 , 0 , 0
-135.325     .04       0  268.34    .033       0 285.299     .04       0
Levee=-1,249.89,8.69,-1,285.46,7.23,Levee 26,Levee 28
Bank Sta=268.34,285.299
XS Rating Curve= 0 ,0
Exp/Cntr=0.3,0.1

Type RM Length L Ch R = 1 ,30.11789,11.075,30.118,12.748
Node Photo=\HecRas Photos\W01.JPG
BEGIN DESCRIPTION:
2008 Survey Section
END DESCRIPTION:
Node Name=W1
XS GIS Cut Line= 3
299804.6222780285379008.73655182299776.3362714195379031.30821366
299771.3556696555379035.28263325
#Sta/Elev= 10
  42.295    8.42  53.085    9.09  59.145    5.53  64.845    5.08  67.795    5.22
  70.155    6.74  73.865     6.6  79.635    8.85  83.555   10.92  84.855   10.98
#Mann= 3 , 0 , 0
  42.295     .04       0  53.085    .033       0  79.635     .04       0
Levee=-1,53.085,9.09,-1,70.16,6.76,,Levee 28
Bank Sta=53.085,79.635
XS Rating Curve= 0 ,0
Exp/Cntr=0.3,0.1

River Reach=Warm Creek      ,US of Noels Pond
Reach XY= 30
304728.0455160185381575.99489331304394.4146444975381314.53918168
304282.0890645445381038.74403431304172.1533905495380955.57530702
304243.8505692435380844.68367064304199.3983184535380807.87911891
 304209.435923475380763.90484932304274.4413654855380705.59114398
304241.9386444785380495.27941981 304209.435923475380441.74552638
304156.8579924285380451.30515021304136.3048012025380397.77125679
304101.412174239 5380424.5382035304103.802080194 5380342.3254386
 304061.739735365380256.76680535303914.0435472545380149.22103732
303933.6407760975380091.86329436 303882.97476982 5379963.7643351
 303805.541816835379958.98452318303756.7877353195380016.82024733
303655.4557227665379935.56344481303639.6823434545379869.60204041
303591.8842243245379845.22499966 303519.709064445379879.16166424
303516.8411772925379815.11218461303447.5339045565379796.47091815
303255.3854656575379828.97363915303198.0277227035379755.84251689
303216.6689891635379685.10130057303157.6236630715379656.71209144
Reach Downstream Storage Area=Noel's Pond

Type RM Length L Ch R = 1 ,7941.430,386.999,353.465,357.514
BEGIN DESCRIPTION:
1996 Survey Section (637.00)
END DESCRIPTION:
Node Name=W36
XS GIS Cut Line= 5
304627.1320575995381301.54642526304566.7204908375381331.13175373
304546.9628678035381340.80764526 304445.478595455381390.50749073
304424.8333826395381400.61806119
#Sta/Elev= 24
       0      42  32.322  40.372  33.028      40  41.235    38.8  48.176  37.886
  59.951      36  61.012   35.54   65.81      34  93.021  33.459 119.874  32.806
 142.308      32 155.867    33.7 159.267   32.84 163.167   32.72 172.867   32.04
 177.067    32.4 177.367   33.19 186.767   35.14 190.567   37.74 194.667   40.14
 197.867   41.29 208.738  41.471 213.159      42 225.255  42.463
#Mann= 3 , 0 , 0
       0      .1       0 155.867    .035       0 177.367      .1       0
Bank Sta=155.867,177.367
XS Rating Curve= 0 ,0
Exp/Cntr=0.3,0.1

Type RM Length L Ch R = 1 ,7587.965,139.047,231.748,232.266
Node Photo=\HecRas Photos\W35.JPG
BEGIN DESCRIPTION:
1996 Survey Section (636.00)
END DESCRIPTION:
Node Name=W35
XS GIS Cut Line= 6
305358.2821172365380582.91070243 304705.023525735380890.37974579
304533.4119525235380971.15211821304474.6228942855380998.82234824
304207.6876949385381124.46066585304148.8500944915381152.15374324
#Sta/Elev= 30
    -722   45.72    -579   30.48     -35      30     -26      32      -6      32
       0  29.856  254.6728.86302  279.67   29.22  339.67   29.55  369.67    30.2
  399.67   30.22  409.57   29.76  422.17   30.12  424.17   31.15  426.77   29.49
  435.57   29.21  442.27   29.53  444.07   30.29  519.67    30.3  528.07   29.65
  532.77   30.42  535.07   29.85  537.67   30.09  546.87   35.08  549.67   35.03
 552.282      38 555.226      40 589.872  39.008 598.738      36 614.699  34.171
#Mann= 3 , 0 , 0
    -722      .1       0  424.17    .035       0  444.07      .1       0
Levee=-1,424.64,31.14,-1,459.42,30.39,Levee 29,Levee 30
Bank Sta=424.17,444.07
XS Rating Curve= 0 ,0
Exp/Cntr=0.3,0.1

Type RM Length L Ch R = 1 ,7356.217,152.634,293.905,226.352
BEGIN DESCRIPTION:
1996 Survey Section (635.00)
END DESCRIPTION:
Node Name=W34
XS GIS Cut Line= 6
305398.0686642065380842.93253036304833.9876987025380875.14532837
304212.0330069615380910.66310345304158.571973963 5380913.7160862
304063.5318289745380919.14351449303880.6168932825380929.58918139
#Sta/Elev= 30
    -565   45.72    -335   30.48       0    24.7  47.689  24.776  59.693      30
  69.034      32  93.784  31.986 108.302      28 356.614  27.261 522.707      28
  574.66  27.575 576.039  27.172 622.968   29.09 632.968   28.99 634.768   28.09
 685.668   27.68 700.368      27 710.468   27.55 715.668      27 717.668   27.29
 719.568   28.84 729.568   28.57 733.168   30.32 737.668   33.77 756.423  35.066
 768.363      40 774.245  40.898 797.903  39.222 820.931      32 920.881  30.482
#Mann= 3 , 0 , 0
    -565      .1       0 685.668    .035       0 719.568      .1       0
Levee=-1,95.24,32.1,-1,773.18,40.87,Levee 29,Levee 30
Bank Sta=685.668,719.568
XS Rating Curve= 0 ,0
Exp/Cntr=0.3,0.1

Type RM Length L Ch R = 1 ,7062.312,98.8,118.591,118.374
BEGIN DESCRIPTION:
1996 Survey Section (634.00)
END DESCRIPTION:
Node Name=W33
XS GIS Cut Line= 6
305333.0438583175380909.52089663304696.3669127075380791.82047857
304662.8587991295380785.62594144303897.0440186815380644.05222747
303855.7319983815380636.41500722 302939.523546065380467.03849911
#Sta/Elev= 30
    -508   45.72    -261   30.48 374.176      26 498.255   25.95 540.255   26.18
 542.855   26.23 545.455   27.22 549.455   25.75 551.955    26.1 553.655   25.87
 558.255   25.71 562.755   25.87 572.555   26.71 575.455   25.72 582.155   25.72
 586.855    26.9 588.255   26.92 618.255   25.73 648.255   26.55 728.255   25.96
 938.044  26.018 949.793  27.934 960.267  28.553    1548      26    1738      26
    1747      28    1763      30    1781      32    1792      34    1892      36
#Mann= 3 , 0 , 0
    -508      .1       0 545.455    .035       0 648.255      .1       0
Levee=-1,546.2,27.22,-1,648.255,26.55,Levee 29,Levee 30
Bank Sta=545.455,648.255
XS Rating Curve= 0 ,0
Exp/Cntr=0.3,0.1

Type RM Length L Ch R = 1 ,6960.092,20,17,20
BEGIN DESCRIPTION:
Interpolated Section
END DESCRIPTION:
Node Name=W32a
XS GIS Cut Line= 6
305373.6559004795380882.48947054304712.074591214 5380729.6785703
304119.1947861295380592.73622402303220.1484616945380385.07606707
302975.5874770035380328.58779601302965.8440114775380326.33726728
#Sta/Elev= 27
   -1018   45.72    -894   30.48    -339      28    -308      26       0   26.27
   88.67   26.45  113.04   26.44  117.06   25.87  117.14   23.87  123.31   24.37
  125.17   24.85  128.11   24.93  135.03   24.46  137.54   25.69   143.1   26.16
  193.36   25.97  265.38   26.23     397      26     898      26     953      26
     981      26    1179      28    1375      30    1387      30    1415      32
    1430      34    1440      36
#Mann= 3 , 0 , 0
   -1018      .1       0  113.04    .035       0   143.1      .1       0
Bank Sta=113.04,143.1
XS Rating Curve= 0 ,0
Exp/Cntr=0.5,0.3

Type RM Length L Ch R = 3 ,6957    ,,,
Node Photo=\HecRas Photos\Rt 460 Bridge.JPG
BEGIN DESCRIPTION:
Route 460 Bridge
END DESCRIPTION:
Bridge Culvert--1,0,-1,-1, 0
Deck Dist Width WeirC Skew NumUp NumDn MinLoCord MaxHiCord MaxSubmerge Is_Ogee
3,8,1.6,0, 6, 6, , , 0.98, 0, 1,1,,
    -500  117.93  117.93  135.33  135.33    1200
   26.75   26.75   26.75   26.75   26.75   26.75
       0       0   25.74   25.74       0       0
       0     557     557   574.4   574.4    1500
   26.75   26.75   26.75   26.75   26.75   26.75
       0       0   25.74   25.74       0       0
Pier Skew, UpSta & Num, DnSta & Num=  ,126.63, 2 ,565.7, 2 , 0 , 0 , 0 ,,
       1       1
       0   25.74
       1       1
       0   25.74
BR Coef=-1 , 0 , 0 ,, 0 ,,,0.8,-1,,0,
WSPro=,,,, 1 ,,,, 0 ,,,, 0 ,,,,-1 ,-1 ,-1 , 0 , 0 , 0 , 0 , 0
BC Design=,, 0 ,, 0 ,,,,,,
BC Use User HTab Curves=0
BC User HTab FreeFlow(D)= 0

Type RM Length L Ch R = 1 ,6943.722,123.195,76.783,97.272
Node Photo=\HecRas Photos\W32.JPG
BEGIN DESCRIPTION:
2008 Survey Section
END DESCRIPTION:
Node Name=W32
XS GIS Cut Line= 5
304755.0624568345380723.86703864304394.7057797725380640.62571343
304113.6268121875380575.69730433303378.2603340355380405.82982565
303237.1540776855380373.23469832
#Sta/Elev= 30
  69.221      28  84.092  27.819  89.477      26 199.772  26.299 259.117      26
 552.107   26.44 556.127   25.87 556.207   23.87 562.377   24.37 564.237   24.85
 567.177   24.93 574.097   24.46 576.607   25.69 582.167   26.16 632.427   25.97
 704.447   26.23 724.712  25.997 843.703  25.842   881.5  24.815 894.381  24.563
 906.814      24 937.905  24.113 960.636   24.66 983.982  24.6711066.262  25.407
1123.327  25.5491186.665      261428.444  26.4091459.178  27.243    1604      28
#Mann= 3 , 0 , 0
  69.221      .1       0 552.107    .035       0 582.167      .1       0
Levee=0,,,-1,704.35,26.23,,Levee 31
Bank Sta=552.107,582.167
XS Rating Curve= 0 ,0
Exp/Cntr=0.5,0.3

Type RM Length L Ch R = 3 ,6931.57 ,,,
Node Photo=\HecRas Photos\Rt 460 Rail.JPG
BEGIN DESCRIPTION:
Route 460 Railway Trestle
END DESCRIPTION:
Bridge Culvert--1,0,-1,-1, 0
Deck Dist Width WeirC Skew NumUp NumDn MinLoCord MaxHiCord MaxSubmerge Is_Ogee
12.15,3.65,1.6,0, 6, 6, , , 0.98, 0, 1,1,,
       0     554     554  581.15  581.15    1500
      27      27      27      27      27      27
       0       0    26.7    26.7       0       0
  423.11     560     560  587.15  587.15    1300
      27      27      27      27      27      27
       0       0    26.7    26.7       0       0
BR Coef=-1 , 0 , 0 ,, 0 ,,,0.8,-1,,0,
WSPro=,,,, 1 ,,,, 0 ,,,, 0 ,,,,-1 ,-1 ,-1 , 0 , 0 , 0 , 0 , 0
BC Design=,, 0 ,, 0 ,,,,,,
BC Use User HTab Curves=0
BC User HTab FreeFlow(D)= 0
