HEC-RAS study Blanche_Brook.prj: Stephenville Model

--- Blanche_Brook.g05 (geometry) --- (continued)

Type RM Length L Ch R = 1 ,1375.933,115.399,110.024,80.619
BEGIN DESCRIPTION:
2008 Survey Section
END DESCRIPTION:
Node Name=W15
XS GIS Cut Line= 4
300438.6961542185379587.56423744300439.2666163955379626.41905013
300439.5602225855379646.41689395300441.2129295155379758.98459923
#Sta/Elev= 19
     -31      24     -29      22     -27      20     -22      18   -1.41   17.37
   7.859   17.06   17.61   17.33  31.149    17.5   40.32   18.34  40.369   18.33
  42.579   16.65  45.689   16.82   47.32   17.21  50.709    17.5  53.859   18.77
  69.739   18.84  71.709   19.72  94.129   20.07 140.439   20.75
#Mann= 3 , 0 , 0
     -31      .1       0   40.32    .045       0  53.859      .1       0
Bank Sta=40.32,53.859
XS Rating Curve= 0 ,0
Exp/Cntr=0.3,0.1

Type RM Length L Ch R = 1 ,1265.909,88.883,82.766,73.503
BEGIN DESCRIPTION:
Interpolated Section
END DESCRIPTION:
Node Name=W14a
XS GIS Cut Line= 3
300370.6541418085379721.89731956300384.7266877325379740.56782603
300435.0195849435379807.29305599
#Sta/Elev= 21
    11.9      22   18.49      20   30.14      18   35.28  17.705  46.005  17.259
  48.973  16.967  51.589  16.845  54.394  16.982   55.05   16.66   57.68   16.43
   59.67    16.5  61.031  16.606  62.371  16.776  64.352  17.391  65.938  17.451
  74.342  17.963  74.403  17.986  75.581    18.6   83.57  20.416  89.684  20.476
 118.816  20.744
#Mann= 3 , 0 , 0
    11.9      .1       0  54.394    .045       0  64.352      .1       0
Levee=-1,54.46,16.97,0,,,,
Bank Sta=54.394,64.352
XS Rating Curve= 0 ,0
Exp/Cntr=0.3,0.1

Type RM Length L Ch R = 1 ,1183.143,20.173,34.556,39.04
BEGIN DESCRIPTION:
2008 Survey Section
END DESCRIPTION:
Node Name=W14
XS GIS Cut Line= 3
300298.9502244315379806.31093566300374.6881692135379826.69472821
300419.7251011965379838.81577904
#Sta/Elev= 12
   -52.1      20   -23.4      18  26.333   18.19  31.403   17.15  34.043   16.05
  35.983   15.93  38.723   15.93  40.823   16.15  43.553   16.45  48.263   17.31
  53.363   20.79  72.973   20.74
#Mann= 3 , 0 , 0
   -52.1      .1       0  31.403    .045       0  48.263      .1       0
Bank Sta=31.403,48.263
XS Rating Curve= 0 ,0
Exp/Cntr=0.3,0.1

Type RM Length L Ch R = 1 ,1125.215,33.473,35.913,35.28
BEGIN DESCRIPTION:
2008 Survey Section
END DESCRIPTION:
Node Name=W13
XS GIS Cut Line= 4
300347.5260179465379785.28417287 300347.485885715379786.86366303
300346.4538013975379827.48355279300344.3981726435379908.38722733
#Sta/Elev= 15
  -18.58      22  -11.33      20   11.07      18  23.633   18.01  28.263   16.93
  38.363   17.21  41.873   15.87  46.323   15.59  54.453   15.93   56.92   17.21
  59.033   18.41  71.663   18.51  89.513   19.07 102.033   19.32 104.563   19.79
#Mann= 3 , 0 , 0
  -18.58      .1       0  38.363    .045       0   56.92      .1       0
Levee=-1,38.24,17.21,0,,,,
Bank Sta=38.363,56.92
XS Rating Curve= 0 ,0
Exp/Cntr=0.3,0.1

Type RM Length L Ch R = 1 ,1051.997,119.597,121.94,125.44
BEGIN DESCRIPTION:
2008 Survey Section
END DESCRIPTION:
Node Name=W12
XS GIS Cut Line= 2
300278.1797119045379817.14976326300273.9853621615379862.86817545
#Sta/Elev= 13
  41.591   23.68  49.111   18.69  53.161   18.16  58.451   16.07   61.74   16.07
  64.511   15.87   67.45   15.87  69.241   15.73   70.34   16.31  71.881   17.03
  81.081   18.05  84.021   19.03  87.501   19.15
#Mann= 3 , 0 , 0
  41.591     .04       0  53.161    .045       0  71.881     .04       0
Bank Sta=53.161,71.881
XS Rating Curve= 0 ,0
Exp/Cntr=0.3,0.1

Type RM Length L Ch R = 1 ,802.9447,71.609,75.267,71.522
BEGIN DESCRIPTION:
2008 Survey Section
END DESCRIPTION:
Node Name=W11
XS GIS Cut Line= 2
 300109.024391465379677.44797171300053.624571032 5379697.0932981
#Sta/Elev= 14
  52.439   19.05  60.639   13.67  67.509   12.77   70.92    12.8  74.999   12.75
   77.01   12.66  78.429   12.53   79.67   12.67  81.389   12.61  82.689   12.83
  86.889   14.84  90.719   14.58 105.649   15.24 111.219   15.91
#Mann= 3 , 0 , 0
  52.439     .04       0  60.639    .045       0  82.689     .04       0
Levee=0,,,-1,86.82,14.83,,
Bank Sta=60.639,82.689
XS Rating Curve= 0 ,0
Exp/Cntr=0.3,0.1

Type RM Length L Ch R = 1 ,727.6773,79.11,78.888,80.462
BEGIN DESCRIPTION:
Interpolated Section
END DESCRIPTION:
Node Name=W10a
XS GIS Cut Line= 2
300099.889136565 5379608.0488858300038.2185467355379634.14028919
#Sta/Elev= 20
  50.773   18.02   57.42  15.077  58.467   14.96  62.989   13.48  69.061  11.985
  70.106  11.687   71.81   11.63   73.84    11.6   75.81   11.64  77.044  11.675
  77.804  11.749  81.308  12.491  83.682  13.531  86.819  14.279  89.043  13.666
  91.899  12.995  97.556  13.624  109.94  13.945 114.019  14.165 117.736  14.562
#Mann= 3 , 0 , 0
  50.773     .04       0  62.989    .045       0  83.682     .04       0
Levee=0,,,-1,86.88,14.29,,
Bank Sta=62.989,83.682
XS Rating Curve= 0 ,0
Exp/Cntr=0.3,0.1

Type RM Length L Ch R = 1 ,648.7893,69.05,68.73,68.507
BEGIN DESCRIPTION:
2008 Survey Section
END DESCRIPTION:
Node Name=W10
XS GIS Cut Line= 2
300092.3868587025379526.86943979300002.014689702   5379565.73747
#Sta/Elev= 18
  44.297   16.94  50.107   16.49   56.85      12  58.897   10.66   59.71   10.53
  60.207   10.33   61.09    10.5  62.927   10.43   64.42    10.6  66.967   10.56
   68.04   10.78  72.507   10.88   74.47   11.73  79.667   13.85  86.267   11.24
  93.617   12.34 115.007   12.67 119.837   13.15
#Mann= 3 , 0 , 0
  44.297     .04       0   56.85    .045       0   74.47     .04       0
Levee=0,,,-1,79.82,13.84,,
Bank Sta=56.85,74.47
XS Rating Curve= 0 ,0
Exp/Cntr=0.3,0.1

Type RM Length L Ch R = 1 ,580.0592,74.519,73.956,72.988
BEGIN DESCRIPTION:
Interpolated Section
END DESCRIPTION:
Node Name=W9a
XS GIS Cut Line= 2
300073.6423346195379462.06826613299999.8798686985379497.88561736
#Sta/Elev= 27
  49.643   14.19  54.069  13.688  55.739  13.612  61.845  11.566  63.644  10.018
   64.55    9.82  64.963   9.522  66.338   9.285   67.81    9.35  69.317   9.354
  69.594    9.36   70.43    9.51  72.035   9.585   72.61    9.82  73.741    9.96
  77.476  10.826  79.808  10.866   87.65  12.327  91.386   11.59  94.878  11.015
  98.263   11.33 102.927  11.637 107.819  11.648 111.971   11.38 114.559  11.722
 126.353  11.921 131.642   12.22
#Mann= 3 , 0 , 0
  49.643     .04       0  61.845    .045       0  79.808     .04       0
Levee=0,,,-1,87.75,12.34,,
Ice Thickness=0.15,0.15,0.15
Ice Mann=0.04,0.04,0.04
Ice Specific Gravity=0.916
Ice Is Channel=-1
Ice Is OB= 0
Ice Friction Angle=45
Ice Porosity=0
Ice K1=0.33
Ice Max Mean Vel=1.524
Ice Cohesion=0
Ice Fixed Mann=-1
Bank Sta=61.845,79.808
XS Rating Curve= 0 ,0
Exp/Cntr=0.3,0.1

Type RM Length L Ch R = 1 ,506.1030,11.553,11.974,12.929
BEGIN DESCRIPTION:
2008 Survey Section
END DESCRIPTION:
Node Name=W9
XS GIS Cut Line= 2
300056.1398469045379388.59785433299980.8645969775379435.98704577
#Sta/Elev= 16
  17.605   11.23  22.255   10.54  30.425   10.42  32.315    8.43    33.7    8.34
  35.145    8.16  38.705     8.2      40    8.48  41.375    8.59  47.325    10.9
  62.535   10.61  70.055   10.93  80.505   10.83  85.045   10.21  87.875   10.88
 106.555   11.22
#Mann= 3 , 0 , 0
  17.605     .04       0  30.425    .045       0  47.325     .04       0
Levee=0,,,-1,47.37,10.91,,
Ice Thickness=0.15,0.15,0.15
Ice Mann=0.04,0.04,0.04
Ice Specific Gravity=0.916
Ice Is Channel=-1
Ice Is OB= 0
Ice Friction Angle=45
Ice Porosity=0
Ice K1=0.33
Ice Max Mean Vel=1.524
Ice Cohesion=0
Ice Fixed Mann=-1
Bank Sta=30.425,47.325
XS Rating Curve= 0 ,0
Exp/Cntr=0.3,0.1

Type RM Length L Ch R = 1 ,494.1285,15.27,14.846,14.427
BEGIN DESCRIPTION:
2008 Survey Section
END DESCRIPTION:
Node Name=W8
XS GIS Cut Line= 4
300090.8916212315379368.46471498300058.5959418035379379.98234975
299964.7175778395379413.46226807299937.0287000835379423.33697537
#Sta/Elev= 19
       0  12.547  14.348  12.252  21.386      12  26.323  11.318  34.288   11.05
  43.138   10.47  55.978   10.64  57.898     9.9  58.348    7.99  67.408    8.16
  67.688    9.87  69.908   10.63  82.668   10.75  98.548   10.55 110.268   10.82
 133.958   11.74  158.33      12 162.957      14 163.355  14.007
#Mann= 3 , 0 , 0
       0     .04       0  55.978    .033       0  69.908     .04       0
Levee=-1,56.09,10.64,0,,,,
#XS Ineff= 2 , 0
       0      58   10.64               0
Permanent Ineff=
       F       F
#Block Obstruct= 2 , 0
       0    60.5      10    65.5       0      10
Ice Thickness=0.15,0.15,0.15
Ice Mann=0.04,0.04,0.04
Ice Specific Gravity=0.916
Ice Is Channel=-1
Ice Is OB= 0
Ice Friction Angle=45
Ice Porosity=0
Ice K1=0.33
Ice Max Mean Vel=1.524
Ice Cohesion=0
Ice Fixed Mann=-1
Bank Sta=55.978,69.908
XS Rating Curve= 0 ,0
Exp/Cntr=0.5,0.3

Type RM Length L Ch R = 3 ,493.61  ,,,
BEGIN DESCRIPTION:
Miss Drive Bridge
END DESCRIPTION:
Bridge Culvert--1,0,-1,-1, 0
Deck Dist Width WeirC Skew NumUp NumDn MinLoCord MaxHiCord MaxSubmerge Is_Ogee
0.52,12.87,1.6,0, 6, 6, , , 0.98, 0, 1,1,,
   55.98    58.4    58.4    67.6    67.6   69.91
   10.64   10.65   10.65   10.65   10.65   10.63
       0       0    9.86    9.86       0       0
   31.34    41.1    41.1    50.3    50.3   57.72
   10.63   10.65   10.65   10.65   10.65   10.63
       0       0    9.86    9.86       0       0
BR Coef=-1 , 0 , 0 ,, 0 ,,,0.8,-1,,0,
WSPro=,,,, 1 ,,,, 0 ,,,, 0 ,,,,-1 ,-1 ,-1 , 0 , 0 , 0 , 0 , 0
BC Design=,, 0 ,, 0 ,,,,,,
BC Use User HTab Curves=0
BC User HTab FreeFlow(D)= 0

Type RM Length L Ch R = 1 ,479.2822,18.024,15.05,14.12
BEGIN DESCRIPTION:
2008 Survey Section
END DESCRIPTION:
Node Name=W7
XS GIS Cut Line= 2
 300049.926581165379364.90465646299964.7605915165379405.41502764
#Sta/Elev= 19
  21.241   10.92  35.011   10.52  38.871   10.42  40.681    9.88  40.941    8.26
  43.581    7.91   45.45    7.87  46.641    7.75   48.62    7.74  49.941    7.45
   50.16    7.77  50.851    8.09  50.991    9.91  53.231   10.52  62.391   10.75
  80.321   10.49  84.271    9.94  93.421   10.73 115.551   11.48
#Mann= 3 , 0 , 0
  21.241     .04       0  38.871    .045       0  53.231     .04       0
Levee=0,,,-1,62.47,10.76,,
Bank Sta=38.871,53.231
XS Rating Curve= 0 ,0
Exp/Cntr=0.5,0.3

Type RM Length L Ch R = 1 ,464.2327,69.028,69.847,71.832
BEGIN DESCRIPTION:
2008 Survey Section
END DESCRIPTION:
Node Name=W6
XS GIS Cut Line= 2
300055.7657332375379338.69292146299958.817893427 5379403.0048548
#Sta/Elev= 17
   22.96   10.52   48.73    9.51   58.75    9.58   61.23     7.8   62.07    7.61
   64.51    7.57   65.54    7.39    68.8    7.37   70.02    7.56   72.83     7.6
   74.24    8.01      75   10.17   89.75   10.61   97.32   10.52  101.53    9.83
  114.83   10.76   139.3   11.54
#Mann= 3 , 0 , 0
   22.96     .04       0   58.75     .03       0      75     .04       0
Bank Sta=58.75,75
XS Rating Curve= 0 ,0
Exp/Cntr=0.3,0.1

Type RM Length L Ch R = 1 ,394.3861,63.972,68.222,69.71
BEGIN DESCRIPTION:
Interpolated Section
END DESCRIPTION:
Node Name=W5a
XS GIS Cut Line= 3
300115.5698633285379255.65033573300033.2517324575379284.08258489
299946.5794008885379314.01875205
#Sta/Elev= 26
     -19      10      19       8   68.09   9.179  89.294   8.613  90.275   8.614
   92.44   8.982  97.539   9.115   99.58    8.28 101.469   8.242 102.279   7.974
  102.84    7.36 104.951   7.203 106.812   7.024  109.37    7.27  110.62   8.384
 110.902   8.395 118.994   8.601 121.899   8.582 122.526   8.561 124.614   8.717
 127.687   9.281  128.75    9.36 130.906   9.161 141.076   9.734 152.738  10.105
 159.787  10.579
#Mann= 3 , 0 , 0
     -19     .04       0  97.539    .033       0 127.687     .04       0
Levee=-1,97.68,9.12,-1,128.75,9.36,,
Bank Sta=97.539,127.687
XS Rating Curve= 0 ,0
Exp/Cntr=0.3,0.1

Type RM Length L Ch R = 1 ,326.1642,14.443,16.892,18.313
BEGIN DESCRIPTION:
2008 Survey Section
END DESCRIPTION:
Node Name=W5
XS GIS Cut Line= 5
300276.8093800145379170.68468354300136.6980384355379199.28209533
300009.1614444545379225.31293948299892.9600124975379249.03022148
299881.1651905175379251.43760248
#Sta/Elev= 19
    -163      12     -20      10      34       8 110.166    7.87 127.686    7.73
 129.396    8.44 136.526    8.83 139.276    6.85 140.746     6.5 143.606    6.65
 149.266    6.75 151.736    6.57 153.196    6.91 156.066    8.46 172.866    8.99
 177.796    9.64  183.93      10 188.262  11.446 189.834      12
#Mann= 3 , 0 , 0
    -163     .04       0 136.526    .033       0 156.066     .04       0
Levee=-1,136.5,8.84,0,,,,
Bank Sta=136.526,156.066
XS Rating Curve= 0 ,0
Exp/Cntr=0.3,0.1

Type RM Length L Ch R = 1 ,309.2723,15.642,14.996,14.953
BEGIN DESCRIPTION:
2008 Survey Section
END DESCRIPTION:
Node Name=W4
XS GIS Cut Line= 4
300136.303502507 5379189.7286179300007.384630526  5379210.427634
 299915.888196465379225.11816094299805.3834867285379242.86062743
#Sta/Elev= 15
      -8      10      44       8  122.57    8.66  141.46    8.73  143.48    9.36
  148.05    9.22  150.25    8.58  152.14    6.77  154.09     6.4  158.69    6.59
  165.12    6.64  169.24    8.59  176.97    9.14  202.08    9.12     314      10
#Mann= 3 , 0 , 0
      -8     .04       0  148.05    .033       0  176.97     .04       0
Levee=-1,143.55,9.35,0,,,,
#XS Ineff= 2 , 0
       0     151    9.36     168       0    9.14
Permanent Ineff=
       F       F
Bank Sta=148.05,176.97
XS Rating Curve= 0 ,0
Exp/Cntr=0.5,0.3

Type RM Length L Ch R = 3 ,305.02  ,,,
BEGIN DESCRIPTION:
Carolina Ave Bridge
END DESCRIPTION:
Bridge Culvert--1,0,-1,-1, 0
Deck Dist Width WeirC Skew NumUp NumDn MinLoCord MaxHiCord MaxSubmerge Is_Ogee
4.25,8.94,1.6,0, 6, 6, , , 0.98, 0, 1,1,,
  143.48     155     155   163.9   163.9  176.97
    9.36    9.55    9.55    9.55    9.55    9.14
       0       0    8.55    8.55       0       0
  214.21     234     234   242.9   242.9  251.75
     9.3    9.55    9.55    9.55    9.55    9.29
       0       0    8.55    8.55       0       0
BR Coef=-1 , 0 , 0 ,, 0 ,,,0.8,-1,,0,
WSPro=,,,, 1 ,,,, 0 ,,,, 0 ,,,,-1 ,-1 ,-1 , 0 , 0 , 0 , 0 , 0
BC Design=,, 0 ,, 0 ,,,,,,
BC Use User HTab Curves=0
BC User HTab FreeFlow(D)= 0

Type RM Length L Ch R = 1 ,294.2762,85.792,40.217,25.479
BEGIN DESCRIPTION:
2008 Survey Section
END DESCRIPTION:
Node Name=W3
XS GIS Cut Line= 2
300028.4277358875379191.25291856299923.975984997 5379209.3649225
#Sta/Elev= 10
 202.728    9.01 214.208     9.3 228.308    9.24 232.428    6.66 237.808    6.42
 240.768    6.38 243.528     6.8 247.008       9 251.748    9.29 287.538    8.72
#Mann= 3 , 0 , 0
 202.728     .04       0 228.308    .033       0 247.008     .04       0
Levee=-1,214.22,9.3,-1,251.63,9.29,,
#XS Ineff= 2 , 0
       0     233     9.3   243.3       0    9.29
Permanent Ineff=
       F       F
Bank Sta=228.308,247.008
XS Rating Curve= 0 ,0
Exp/Cntr=0.5,0.3

Type RM Length L Ch R = 1 ,254.0591,74.46,106.674,110.065
BEGIN DESCRIPTION:
2008 Survey Section
END DESCRIPTION:
Node Name=W2
XS GIS Cut Line= 6
300215.3837418395378846.99193121299986.9183204945379124.95448985
299918.8401838145379207.78178576299916.7070083875379210.37711461
299916.1888667195379211.00751191 299838.846335575379305.10633824
#Sta/Elev= 19
     -68      10      44       8      89       6     241       6 291.805    7.08
 331.375    7.29 339.445    8.51 343.725    8.55 346.775    6.59 348.565    6.16
 349.185    5.86 351.425    5.95 353.245    6.12 354.635    6.44 357.715    7.91
 365.735    7.56 380.705       8 403.195    8.85     525      10
#Mann= 3 , 0 , 0
     -68     .04       0 343.725    .033       0 357.715     .04       0
Levee=-1,343.89,8.55,-1,357.71,7.92,,
Bank Sta=343.725,357.715
XS Rating Curve= 0 ,0
Exp/Cntr=0.3,0.1

Type RM Length L Ch R = 1 ,147.3854,137.703,117.268,115.163
BEGIN DESCRIPTION:
Interpolated Section
END DESCRIPTION:
Node Name=W1a
XS GIS Cut Line= 2
299915.6107996985379079.12916934299831.1880560285379131.14722352
#Sta/Elev= 22
 234.475   7.718  249.89    8.69 262.604   6.815 264.954   6.713  268.34    7.02
  268.37    7.02 271.383   6.978 273.551   5.906 274.823   5.655 275.264   5.488
 276.833   5.554 278.107   5.659  279.08   5.838 280.839   6.487 281.236   6.693
 285.299    7.22 286.852   7.155  292.31   7.223 297.333   7.827 303.214   8.571
 310.622   9.767 313.079   9.865
#Mann= 3 , 0 , 0
 234.475     .04       0  268.34    .033       0 285.299     .04       0
Levee=-1,249.89,8.69,-1,285.46,7.23,,
Bank Sta=268.34,285.299
XS Rating Curve= 0 ,0
Exp/Cntr=0.3,0.1

Type RM Length L Ch R = 1 ,30.11789,11.075,30.118,12.748
BEGIN DESCRIPTION:
2008 Survey Section
END DESCRIPTION:
Node Name=W1
XS GIS Cut Line= 3
299804.6222780285379008.73655182299776.3362714195379031.30821366
299771.3556696555379035.28263325
#Sta/Elev= 10
  42.295    8.42  53.085    9.09  59.145    5.53  64.845    5.08  67.795    5.22
  70.155    6.74  73.865     6.6  79.635    8.85  83.555   10.92  84.855   10.98
#Mann= 3 , 0 , 0
  42.295     .04       0  53.085    .033       0  79.635     .04       0
Levee=0,,,-1,70.16,6.76,,
Bank Sta=53.085,79.635
XS Rating Curve= 0 ,0
Exp/Cntr=0.3,0.1

River Reach=Warm Creek      ,US of Noels Pond

Type RM Length L Ch R = 1 ,7587.965,139.047,231.748,232.266
BEGIN DESCRIPTION:
1996 Survey Section (636.00)
END DESCRIPTION:
Node Name=W35
XS GIS Cut Line= 6
305358.2821172365380582.91070243 304705.023525735380890.37974579
304533.4119525235380971.15211821304474.6228942855380998.82234824
304207.6876949385381124.46066585304148.8500944915381152.15374324
#Sta/Elev= 30
    -722   45.72    -579   30.48     -35      30     -26      32      -6      32
       0  29.856  254.6728.86302  279.67   29.22  339.67   29.55  369.67    30.2
  399.67   30.22  409.57   29.76  422.17   30.12  424.17   31.15  426.77   29.49
  435.57   29.21  442.27   29.53  444.07   30.29  519.67    30.3  528.07   29.65
  532.77   30.42  535.07   29.85  537.67   30.09  546.87   35.08  549.67   35.03
 552.282      38 555.226      40 589.872  39.008 598.738      36 614.699  34.171
#Mann= 3 , 0 , 0
    -722      .1       0  424.17    .035       0  444.07      .1       0
Levee=-1,424.64,31.14,-1,459.42,30.39,,
Bank Sta=424.17,444.07
XS Rating Curve= 0 ,0
Exp/Cntr=0.3,0.1

Type RM Length L Ch R = 1 ,7356.217,152.634,293.905,226.352
BEGIN DESCRIPTION:
1996 Survey Section (635.00)
END DESCRIPTION:
Node Name=W34
XS GIS Cut Line= 6
305398.0686642065380842.93253036304833.9876987025380875.14532837
304212.0330069615380910.66310345304158.571973963 5380913.7160862
304063.5318289745380919.14351449303880.6168932825380929.58918139
#Sta/Elev= 30
    -565   45.72    -335   30.48       0    24.7  47.689  24.776  59.693      30
  69.034      32  93.784  31.986 108.302      28 356.614  27.261 522.707      28
  574.66  27.575 576.039  27.172 622.968   29.09 632.968   28.99 634.768   28.09
 685.668   27.68 700.368      27 710.468   27.55 715.668      27 717.668   27.29
 719.568   28.84 729.568   28.57 733.168   30.32 737.668   33.77 756.423  35.066
 768.363      40 774.245  40.898 797.903  39.222 820.931      32 920.881  30.482
#Mann= 3 , 0 , 0
    -565      .1       0 685.668    .035       0 719.568      .1       0
Levee=-1,95.24,32.1,-1,773.18,40.87,,
Bank Sta=685.668,719.568
XS Rating Curve= 0 ,0
Exp/Cntr=0.3,0.1

Type RM Length L Ch R = 1 ,7062.312,98.8,118.591,118.374
BEGIN DESCRIPTION:
1996 Survey Section (634.00)
END DESCRIPTION:
Node Name=W33
XS GIS Cut Line= 6
305333.0438583175380909.52089663304696.3669127075380791.82047857
304662.8587991295380785.62594144303897.0440186815380644.05222747
303855.7319983815380636.41500722 302939.523546065380467.03849911
#Sta/Elev= 30
    -508   45.72    -261   30.48 374.176      26 498.255   25.95 540.255   26.18
 542.855   26.23 545.455   27.22 549.455   25.75 551.955    26.1 553.655   25.87
 558.255   25.71 562.755   25.87 572.555   26.71 575.455   25.72 582.155   25.72
 586.855    26.9 588.255   26.92 618.255   25.73 648.255   26.55 728.255   25.96
 938.044  26.018 949.793  27.934 960.267  28.553    1548      26    1738      26
    1747      28    1763      30    1781      32    1792      34    1892      36
#Mann= 3 , 0 , 0
    -508      .1       0 545.455    .035       0 648.255      .1       0
Levee=-1,546.2,27.22,-1,649.46,26.55,,
Ice Thickness=0.15,0.15,0.15
Ice Mann=0.04,0.04,0.04
Ice Specific Gravity=0.916
Ice Is Channel=-1
Ice Is OB= 0
Ice Friction Angle=45
Ice Porosity=0
Ice K1=0.33
Ice Max Mean Vel=1.524
Ice Cohesion=0
Ice Fixed Mann=-1
Bank Sta=545.455,648.255
XS Rating Curve= 0 ,0
Exp/Cntr=0.3,0.1

Type RM Length L Ch R = 1 ,6960.092,20,17,20
BEGIN DESCRIPTION:
Interpolated Section
END DESCRIPTION:
Node Name=W32a
XS GIS Cut Line= 6
305373.6559004795380882.48947054304712.074591214 5380729.6785703
304119.1947861295380592.73622402303220.1484616945380385.07606707
302975.5874770035380328.58779601302965.8440114775380326.33726728
#Sta/Elev= 27
   -1018   45.72    -894   30.48    -339      28    -308      26       0   26.27
   88.67   26.45  113.04   26.44  117.06   25.87  117.14   23.87  123.31   24.37
  125.17   24.85  128.11   24.93  135.03   24.46  137.54   25.69   143.1   26.16
  193.36   25.97  265.38   26.23     397      26     898      26     953      26
     981      26    1179      28    1375      30    1387      30    1415      32
    1430      34    1440      36
#Mann= 3 , 0 , 0
   -1018      .1       0  113.04    .035       0   143.1      .1       0
#Block Obstruct= 2 ,-1
     112     120    26.5     130     140    26.5
Ice Thickness=0.15,0.15,0.15
Ice Mann=0.04,0.04,0.04
Ice Specific Gravity=0.916
Ice Is Channel=-1
Ice Is OB= 0
Ice Friction Angle=45
Ice Porosity=0
Ice K1=0.33
Ice Max Mean Vel=1.524
Ice Cohesion=0
Ice Fixed Mann=-1
Bank Sta=113.04,143.1
XS Rating Curve= 0 ,0
Exp/Cntr=0.5,0.3

Type RM Length L Ch R = 3 ,6957    ,,,
BEGIN DESCRIPTION:
Route 460 Bridge
END DESCRIPTION:
Bridge Culvert--1,0,-1,-1, 0
Deck Dist Width WeirC Skew NumUp NumDn MinLoCord MaxHiCord MaxSubmerge Is_Ogee
3,8,1.6,0, 6, 6, , , 0.98, 0, 1,1,,
    -500  117.93  117.93  135.33  135.33    1200
   26.75   26.75   26.75   26.75   26.75   26.75
       0       0   25.74   25.74       0       0
       0     557     557   574.4   574.4    1500
   26.75   26.75   26.75   26.75   26.75   26.75
       0       0   25.74   25.74       0       0
Pier Skew, UpSta & Num, DnSta & Num=  ,126.63, 2 ,565.7, 2 , 0 , 0 , 0 ,,
       1       1
       0   25.74
       1       1
       0   25.74
BR Coef=-1 , 0 , 0 ,, 0 ,,,0.8,-1,,0,
WSPro=,,,, 1 ,,,, 0 ,,,, 0 ,,,,-1 ,-1 ,-1 , 0 , 0 , 0 , 0 , 0
BC Design=,, 0 ,, 0 ,,,,,,
BC Use User HTab Curves=0
BC User HTab FreeFlow(D)= 0

Type RM Length L Ch R = 1 ,6943.722,123.195,76.783,97.272
BEGIN DESCRIPTION:
2008 Survey Section
END DESCRIPTION:
Node Name=W32
XS GIS Cut Line= 5
304755.0624568345380723.86703864304394.7057797725380640.62571343
304113.6268121875380575.69730433303378.2603340355380405.82982565
303237.1540776855380373.23469832
#Sta/Elev= 30
  69.221      28  84.092  27.819  89.477      26 199.772  26.299 259.117      26
 552.107   26.44 556.127   25.87 556.207   23.87 562.377   24.37 564.237   24.85
 567.177   24.93 574.097   24.46 576.607   25.69 582.167   26.16 632.427   25.97
 704.447   26.23 724.712  25.997 843.703  25.842   881.5  24.815 894.381  24.563
 906.814      24 937.905  24.113 960.636   24.66 983.982  24.6711066.262  25.407
1123.327  25.5491186.665      261428.444  26.4091459.178  27.243    1604      28
#Mann= 3 , 0 , 0
  69.221      .1       0 552.107    .035       0 582.167      .1       0
Levee=0,,,-1,704.35,26.23,,
Bank Sta=552.107,582.167
XS Rating Curve= 0 ,0
Exp/Cntr=0.5,0.3

Type RM Length L Ch R = 3 ,6931.57 ,,,
BEGIN DESCRIPTION:
Route 460 Railway Trestle
END DESCRIPTION:
Bridge Culvert--1,0,-1,-1, 0
Deck Dist Width WeirC Skew NumUp NumDn MinLoCord MaxHiCord MaxSubmerge Is_Ogee
12.15,3.65,1.6,0, 6, 6, , , 0.98, 0, 1,1,,
       0     554     554  581.15  581.15    1500
      27      27      27      27      27      27
       0       0    26.7    26.7       0       0
  423.11     560     560  587.15  587.15    1300
      27      27      27      27      27      27
       0       0    26.7    26.7       0       0
BR Coef=-1 , 0 , 0 ,, 0 ,,,0.8,-1,,0,
WSPro=,,,, 1 ,,,, 0 ,,,, 0 ,,,,-1 ,-1 ,-1 , 0 , 0 , 0 , 0 , 0
BC Design=,, 0 ,, 0 ,,,,,,
BC Use User HTab Curves=0
BC User HTab FreeFlow(D)= 0

Type RM Length L Ch R = 1 ,6699.612,174.266,215.182,71.29
BEGIN DESCRIPTION:
1996 Survey Section (631.00)
END DESCRIPTION:
Node Name=W30
XS GIS Cut Line= 4
  304337.34655055380440.25391269303885.2392684315380440.25533154
303835.9968712245380432.22324907303543.9179118895380384.58133028
#Sta/Elev= 30
  279.74      28  296.74      26  396.74    24.9  423.04   24.89  424.04   24.21
  439.34   24.76  440.54   23.82  446.74    21.8  453.04   23.82  453.44   24.21
  454.64   24.59  456.14   24.02  461.44   23.85  462.24   24.17  467.74   24.01
  469.44   25.03  481.74    24.9  571.74    25.6  596.74    26.2  676.74    24.8
 710.405      24 728.945  23.799 729.943      24 891.661  24.779 961.754  25.309
1020.043      261069.432   26.231074.301  27.5211076.224  29.0361077.679  29.856
#Mann= 3 , 0 , 0
  279.74      .1       0  423.04    .035       0  469.44      .1       0
Levee=0,,,-1,597.64,26.19,,
Bank Sta=423.04,469.44
XS Rating Curve= 0 ,0
Exp/Cntr=0.3,0.1

Type RM Length L Ch R = 1 ,6484.431,616.58,562.375,435.815
BEGIN DESCRIPTION:
1996 Survey Section (633.00)
END DESCRIPTION:
Node Name=W29
XS GIS Cut Line= 6
304218.8051609775380263.84443487303882.7370809715380415.61423989
303815.8542459355380406.09868082303776.2530289295380400.46453389
303736.6518119225380394.83038696303716.851203419 5380392.0133135
#Sta/Elev= 28
 662.342   27.16 684.542   27.15 692.342    26.8 699.742   26.74 708.442   25.67
 711.742    26.4 724.842   26.67 736.342   26.65 740.942   25.46 743.242   26.04
 752.342   25.71 777.442    25.8 779.242   24.88 782.342   24.96 787.742   24.62
 797.042   25.06 800.742   25.78 803.742    24.9 808.242   24.75 812.342   24.51
 814.842   24.75 822.842   26.38 824.842   25.61 845.642   25.08 849.642    25.5
 882.842   25.92 962.342   25.961152.342      28
#Mann= 3 , 0 , 0
 662.342      .1       0 777.442    .035       0 822.842      .1       0
Levee=-1,725.54,26.67,0,,,,
Bank Sta=777.442,822.842
XS Rating Curve= 0 ,0
Exp/Cntr=0.3,0.1

Type RM Length L Ch R = 1 ,5922.055,190,176.792,190
BEGIN DESCRIPTION:
1996 Survey Section (629.00)
END DESCRIPTION:
Node Name=W28
XS GIS Cut Line= 4
303806.3940636145379865.06548458303806.3940636145379865.06548459
303807.1977242375380045.09012081303807.7377673825380166.06291441
#Sta/Elev= 30
       0  28.005    4.84  28.099  10.284  27.979  20.749  27.202  26.643  26.969
  28.642  27.036  31.852  26.929  32.783  26.964  33.969  26.865  35.824  26.942
  38.408  26.772  40.159  26.824  41.584  26.752  46.464  26.742  60.071  26.359
   61.26  26.262  67.129  26.159  69.717      26  71.974  25.755  75.361  25.085
  79.394      24    83.9   22.98    84.2   22.62    88.4   22.27    92.4   22.57
      93   23.58     123   23.27     153   23.19     288      24     301      26
#Mann= 3 , 0 , 0
       0      .1       0  79.394    .035       0      93      .1       0
Bank Sta=79.394,93
XS Rating Curve= 0 ,0
Exp/Cntr=0.3,0.1

Type RM Length L Ch R = 1 ,5745.264,259.064,255.295,179.874
BEGIN DESCRIPTION:
1996 Survey Section (629.10)
END DESCRIPTION:
Node Name=W27
XS GIS Cut Line= 6
303897.5228163715379641.80152513303866.3019902455379693.03880746
 303855.895046885379710.11790374303587.1544735345380151.15481206
 303562.709615165380191.27188343303475.6024384215380334.22566015
#Sta/Elev= 25
  93.678      27 113.678      26 173.678      25 233.678    24.9 288.678      25
 391.678      25 392.438    24.4 392.448    22.7  395.22    22.1  398.07    22.1
 400.668    22.7 508.678      25 593.678    25.2 642.678    24.9 835.075  24.758
 842.339  25.047 843.953   25.09 846.085  25.144  850.64  25.351 851.731  25.385
 853.006  25.422 858.585  25.677 862.203  25.834 863.076  25.865  866.08      26
#Mann= 3 , 0 , 0
  93.678      .1       0 391.678     .03       0 508.678      .1       0
Bank Sta=391.678,508.678
XS Rating Curve= 0 ,0
Exp/Cntr=0.3,0.1

Type RM Length L Ch R = 1 ,5225.582,86.513,147.307,158.26
BEGIN DESCRIPTION:
1996 Survey Section (627.00)
END DESCRIPTION:
Node Name=W25
XS GIS Cut Line= 3
303397.6071004285379601.05336699303332.0186180245380036.13714577
303314.6786496865380151.16250803
#Sta/Elev= 30
       0      28  44.896  27.812  76.636      24 101.349  22.678     130   21.77
     190   22.06   221.8   22.57     227   21.06   231.7   22.57   236.7   22.18
     250   22.27   252.5   22.52   260.6    26.8   265.6   28.03   272.3   28.44
     280   31.38   281.2    32.1     286    32.2   288.4   33.13   297.2   33.47
   302.2   32.18   313.3   30.08   326.5   26.69     340    22.5     400    22.5
 491.924    24.4 499.908  25.472 501.669      26 505.808      28 556.325  27.606
#Mann= 3 , 0 , 0
       0      .1       0   221.8     .03       0   231.7      .1       0
Levee=-1,220.56,22.52,-1,297.36,33.5,,
Bank Sta=221.8,231.7
XS Rating Curve= 0 ,0
Exp/Cntr=0.3,0.1

Type RM Length L Ch R = 1 ,5078.275,131.874,182.721,103.016
BEGIN DESCRIPTION:
1996 Survey Section (626.00)
END DESCRIPTION:
Node Name=W24
XS GIS Cut Line= 2
 303352.251843395379637.18626122303130.9721827245379982.34539722
#Sta/Elev= 17
 173.918      28 188.918   25.81 213.918   22.44 338.818   22.44 367.918   22.43
 368.918   22.28 374.918   21.08 380.918   22.28 385.118   25.21 386.418   25.28
  387.22   26.53 387.618   26.56 390.718   25.79 396.218    25.7 403.918    22.8
 568.918    22.8 583.918      30
#Mann= 3 , 0 , 0
 173.918      .1       0 367.918     .03       0 380.918      .1       0
Levee=0,,,-1,387.22,26.51,,
Ice Thickness=0.15,0.15,0.15
Ice Mann=0.04,0.04,0.04
Ice Specific Gravity=0.916
Ice Is Channel=-1
Ice Is OB= 0
Ice Friction Angle=45
Ice Porosity=0
Ice K1=0.33
Ice Max Mean Vel=1.524
Ice Cohesion=0
Ice Fixed Mann=-1
Bank Sta=367.918,380.918
XS Rating Curve= 0 ,0
Exp/Cntr=0.3,0.1

Type RM Length L Ch R = 1 ,4910.798,35,30.793,35
BEGIN DESCRIPTION:
1:2500 Community Mapping Section
END DESCRIPTION:
Node Name=490us
XS GIS Cut Line= 4
 303282.70595662 5379418.2374223303233.2754357335379582.20207694
303174.4464749665379777.34204437303135.1536623475379916.66644125
#Sta/Elev= 11
       0      26      32      24      54      24      72      22     147      22
  220.75   20.18     245    18.6     283    18.6  304.58   21.94     379      24
     491      26
#Mann= 3 , 0 , 0
       0      .1       0     147    .035       0  304.58      .1       0
#Block Obstruct= 3 ,-1
     242     244      22     252     254      22     267     273    21.3
Ice Thickness=0.15,0.15,0.15
Ice Mann=0.04,0.04,0.04
Ice Specific Gravity=0.916
Ice Is Channel=-1
Ice Is OB= 0
Ice Friction Angle=45
Ice Porosity=0
Ice K1=0.33
Ice Max Mean Vel=1.524
Ice Cohesion=0
Ice Fixed Mann=-1
Bank Sta=147,304.58
XS Rating Curve= 0 ,0
Exp/Cntr=0.5,0.3

Type RM Length L Ch R = 2 ,4910.6  ,,,
BEGIN DESCRIPTION:
Route 490 Culverts
END DESCRIPTION:
Bridge Culvert--1,0,-1,-1, 0
Deck Dist Width WeirC Skew NumUp NumDn MinLoCord MaxHiCord MaxSubmerge Is_Ogee
1,20,1.6,0, 11, 11, , , 0.98, 0, 1,1,,
       0  134.37  209.24  274.03  298.69  348.17  393.74  430.23  488.38  519.55
  760.07
   28.23   24.52   25.21   25.54   25.63   25.88   26.07   26.25   26.45   26.64
   27.42
       0       0       0       0       0       0       0       0       0       0
       0
       0  134.37  209.24  274.03  298.69  348.17  393.74  430.23  488.38  519.55
  760.07
   28.23   24.52   25.21   25.54   25.63   25.88   26.07   26.25   26.45   26.64
   27.42
       0       0       0       0       0       0       0       0       0       0
       0
BR Coef=-1 , 0 , 0 ,, 0 ,,,0.8,-1,,0,
WSPro=,,,, 1 ,,,, 0 ,,,, 0 ,,,,-1 ,-1 ,-1 , 0 , 0 , 0 , 0 , 0
Culvert=1,2.2,,30.01,0.024,0.9,1,2,3,20.95,243,20.84,243,Culvert #2  , 0 ,0.5
Culvert Bottom n=0.024
Culvert=1,2.2,,29.76,0.024,0.9,1,2,3,21.23,253,20.8,253,Culvert #3  , 0 ,0.5
Culvert Bottom n=0.024
Culvert=1,5,,25.57,0.024,0.9,1,2,3,18.78,270,18.9,270,Culvert #1  , 0 ,0.5
Culvert Bottom n=0.024
BC Design=,, 0 ,, 0 ,,,,,,
BC Use User HTab Curves=0
BC User HTab FreeFlow(D)= 0

River Reach=Blanche Brook   ,DS of Confluence

Type RM Length L Ch R = 1 ,1727.041,38.425,31.866,27.978
BEGIN DESCRIPTION:
2008 Survey Section
END DESCRIPTION:
Node Name=BB11
XS GIS Cut Line= 3
299807.7864269475378971.57526448299733.2779646595378976.35237414
299727.4708878445378976.72469484
#Sta/Elev= 10
 303.369    7.22 315.899     8.9  327.93    8.47 333.249     5.5 339.929    4.47
 342.059    4.78 357.319    5.44 364.019    7.32 378.319    8.03 383.849   10.28
#Mann= 3 , 0 , 0
 303.369     .04       0  327.93    .042       0 364.019     .03       0
Levee=-1,315.94,8.9,0,,,,
Bank Sta=327.93,364.019
XS Rating Curve= 0 ,0
Exp/Cntr=0.3,0.1

Type RM Length L Ch R = 1 ,1695.175,33,30.247,29.947
BEGIN DESCRIPTION:
Interpolated Section
END DESCRIPTION:
Node Name=BB10a
XS GIS Cut Line= 3
299799.994839391 5378935.1190029299718.8196115125378953.47964996
299706.0696942955378956.36349441
#Sta/Elev= 22
 404.903   6.137 416.601   7.943  422.05   8.299 427.618   8.136 431.047   7.144
 432.799   6.262 436.859   5.025 438.242   4.831 439.036   4.316 442.051    4.53
 451.292   4.861 453.052   4.959 454.256   5.105 454.507   5.165 457.315   5.869
  463.65    6.31 463.783    6.33 473.133   7.376 483.587   7.714 493.374   8.028
 495.906    8.42 501.201   9.305
#Mann= 3 , 0 , 0
 404.903     .04       0 427.618    .042       0 473.133     .03       0
Levee=-1,421.96,8.29,0,,,,
Bank Sta=427.618,473.133
XS Rating Curve= 0 ,0
Exp/Cntr=0.3,0.1

Type RM Length L Ch R = 1 ,1664.927,121.636,111.389,102.212
BEGIN DESCRIPTION:
2008 Survey Section
END DESCRIPTION:
Node Name=BB10
XS GIS Cut Line= 2
299792.9686280485378904.34813455299685.5516430365378933.52707675
#Sta/Elev= 16
 436.966    5.11 452.956    7.93 461.346    7.75 466.766    5.21 468.056    5.05
 468.796    4.17  477.57     4.3 484.466    4.67 486.716    4.81 488.256    5.06
 488.576    5.17 492.166    6.46 500.436    7.15 525.756    7.74 541.506     8.1
 548.276    8.38
#Mann= 3 , 0 , 0
 436.966     .04       0 461.346     .03       0 500.436     .03       0
Levee=-1,453.22,7.93,0,,,,
Bank Sta=461.346,500.436
XS Rating Curve= 0 ,0
Exp/Cntr=0.3,0.1

Type RM Length L Ch R = 1 ,1553.538,157.692,137.863,125.752
BEGIN DESCRIPTION:
Interpolated Section
END DESCRIPTION:
Node Name=BB9a
XS GIS Cut Line= 2
299725.3013170545378807.32741864299630.6613077975378853.32246314
#Sta/Elev= 25
 313.423   5.494 331.152   7.409 338.622   7.479 340.455   6.945 343.196   5.536
 344.489   4.966 346.041    4.42 346.465   4.292 347.895   4.108 348.716   3.567
  354.78    3.62 360.488   3.879 362.178   3.961 363.335   4.103 363.576   4.165
 365.033   4.554 366.273   4.917 372.047   5.434 372.486   5.502 374.064    5.68
 383.993   6.963 391.507   7.141 400.547   7.351 403.339   7.495 408.425   7.826
#Mann= 3 , 0 , 0
 313.423     .04       0 338.622     .03       0 383.993     .03       0
Levee=-1,338.37,7.48,0,,,,
Bank Sta=338.622,383.993
XS Rating Curve= 0 ,0
Exp/Cntr=0.3,0.1

Type RM Length L Ch R = 1 ,1415.675,158.169,140.419,140.146
BEGIN DESCRIPTION:
2008 Survey Section
END DESCRIPTION:
Node Name=BB9
XS GIS Cut Line= 2
299626.2413460285378705.45654513  299570.34668825378755.19468992
#Sta/Elev= 12
 192.244    5.97 220.504     7.1 225.634    4.23 227.084    3.63 228.824    3.22
 231.824    2.82 241.454    2.93 245.594    3.37 246.784     3.8 252.644    6.29
 262.414    6.53 267.064    7.14
#Mann= 3 , 0 , 0
 192.244     .04       0 220.504    .045       0 252.644     .03       0
Levee=-1,220.36,7.1,0,,,,
Bank Sta=220.504,252.644
XS Rating Curve= 0 ,0
Exp/Cntr=0.3,0.1

Type RM Length L Ch R = 1 ,1275.257,168.064,166.177,163.118
BEGIN DESCRIPTION:
Interpolated Section
END DESCRIPTION:
Node Name=BB8a
XS GIS Cut Line= 2
299491.2122140655378643.65235928299425.9659520055378718.40909343
#Sta/Elev= 25
 174.101    6.82 190.812   7.552 204.481   7.644 210.871   5.745 211.531   5.384
 212.689   4.932 212.969     4.8 213.987   4.308  215.33    3.93 217.546   3.358
 219.432   2.986 221.696   2.707   225.6   2.393 228.654   2.498 229.417   3.005
 229.684   3.074 231.131   3.344 234.144   4.465 238.642   4.618 244.249   5.021
  245.86   5.302 248.325   5.793 253.797   6.804 267.029   7.127 273.326    7.55
#Mann= 3 , 0 , 0
 174.101     .04       0 204.481    .045       0 253.797     .03       0
Levee=-1,204.13,7.66,0,,,,
Bank Sta=204.481,253.797
XS Rating Curve= 0 ,0
Exp/Cntr=0.3,0.1

Type RM Length L Ch R = 1 ,1109.079,14.535,35.351,37.238
BEGIN DESCRIPTION:
2008 Survey Section
END DESCRIPTION:
Node Name=BB8
XS GIS Cut Line= 2
299337.5536422835378578.67410541299279.4347148645378692.83831755
#Sta/Elev= 16
      22  7.8266  43.288  8.8167  60.701  8.5196  69.681  3.6886  71.157  3.2922
  71.513  3.1466   72.81  2.5897  74.521   2.447  87.603   1.887  91.603   2.086
  92.603  3.1863  92.952  3.3331  94.847  3.9095  98.793  6.3259 117.365  7.2368
 150.107  8.0342
#Mann= 3 , 0 , 0
      22     .04       0  60.701    .045       0  98.793     .03       0
Levee=-1,43.46,8.8,0,,,,
Bank Sta=60.701,98.793
XS Rating Curve= 0 ,0
Exp/Cntr=0.3,0.1

Type RM Length L Ch R = 1 ,1073.728,15.434,34.878,36.514
BEGIN DESCRIPTION:
Interpolated Section
END DESCRIPTION:
Node Name=BB7a
XS GIS Cut Line= 2
299339.5825045725378565.28433151299234.883828444 5378651.3353084
#Sta/Elev= 30
  10.653   6.238  17.548   6.476  35.468   8.183  36.292   8.208  56.095   8.291
  57.264   8.297  65.243   6.624  68.079   5.063  69.857   4.283  70.285    4.07
  71.847    3.28  72.815   2.929  73.908   2.779  74.331   2.728  74.537   2.664
  75.607   2.398  78.837   1.984  89.664   1.783  92.043   2.125   93.28   2.241
  94.184   2.848    94.5   2.942  95.583   3.195  96.213   3.467  99.781   5.611
 103.502   6.695 111.867   6.996 116.573   7.124  127.67   7.276 146.176   7.997
#Mann= 3 , 0 , 0
  10.653     .04       0  57.264    .045       0 103.502     .03       0
Levee=-1,56.09,8.29,0,,,,
Bank Sta=57.264,103.502
XS Rating Curve= 0 ,0
Exp/Cntr=0.3,0.1

Type RM Length L Ch R = 1 ,1038.850,97.122,98.076,97.578
BEGIN DESCRIPTION:
2008 Survey Section
END DESCRIPTION:
Node Name=BB7
XS GIS Cut Line= 2
299346.6748915995378558.28651821299210.1001466295378600.12819631
#Sta/Elev= 17
 175.444    4.67 183.494    4.88 204.414    7.59 228.494    8.05 239.174    8.27
 248.014    3.33 249.784    3.02 250.024     2.9 251.274    2.41 255.044     1.7
 267.684    1.68 269.814    2.23 272.984     2.7 280.074    6.86 287.564    7.01
 301.714    7.02 318.284    7.96
#Mann= 3 , 0 , 0
 175.444     .04       0 239.174    .036       0 280.074     .03       0
Levee=-1,238.7,8.26,0,,,,
Bank Sta=239.174,280.074
XS Rating Curve= 0 ,0
Exp/Cntr=0.3,0.1

Type RM Length L Ch R = 1 ,940.7740,81.937,84.649,84.827
BEGIN DESCRIPTION:
Interpolated Section
END DESCRIPTION:
Node Name=BB6a
XS GIS Cut Line= 2
299289.5190004735378475.50399297  299176.63230175378507.59647093
#Sta/Elev= 27
   88.93   4.917  94.131   4.978  94.298   4.992 103.705   4.341 107.647   4.436
 108.295     4.4 123.204   4.574 129.424   4.653 130.104   4.659 135.816   2.339
 136.959   2.189 137.114   2.132 137.922   1.901 140.358   1.558 148.524   1.503
 150.956   1.841 154.575   2.183 154.621   2.196 157.665   3.135 162.669   5.293
 162.859   5.332 170.583   5.733 171.219   5.736 182.172   5.714 187.373   5.687
  194.98   5.821  206.29   6.323
#Mann= 3 , 0 , 0
   88.93     .04       0 130.104    .036       0 162.669     .03       0
Levee=-1,130.08,4.68,0,,,,
Bank Sta=130.104,162.669
XS Rating Curve= 0 ,0
Exp/Cntr=0.3,0.1

Type RM Length L Ch R = 1 ,856.1249,20.593,20.052,19.351
BEGIN DESCRIPTION:
2008 Survey Section
END DESCRIPTION:
Node Name=BB6
XS GIS Cut Line= 2
299262.0412684325378398.81673008 299169.088876585378420.15556043
#Sta/Elev= 13
 112.121    5.13 114.951    5.06 119.911    2.22 122.331    1.63 133.471    1.55
 143.541    1.35 150.291    1.74 153.661    2.14 159.411    4.01 167.961    4.64
 180.791    4.59 194.971    4.46 207.491    4.91
#Mann= 3 , 0 , 0
 112.121     .04       0 114.951    .033       0 167.961     .03       0
Levee=0,,,-1,167.98,4.63,,
Bank Sta=114.951,167.961
XS Rating Curve= 0 ,0
Exp/Cntr=0.3,0.1

Type RM Length L Ch R = 1 ,836.0733,22.384,21.424,19.965
BEGIN DESCRIPTION:
Interpolated Section
END DESCRIPTION:
Node Name=BB5a
XS GIS Cut Line= 2
299268.8219511995378376.18757931299134.3559988055378411.67550076
#Sta/Elev= 25
  111.46   5.464   114.7   5.327 117.229   4.595  120.38   3.778 123.151    3.47
 129.445   3.442 135.907   3.531 138.226    3.55 142.215   2.223  146.76   1.448
 147.438   1.118 150.789   1.238  158.32   1.599 160.976   1.778 163.752   1.815
 165.493   1.954 172.955   4.308 173.022   4.315   186.4   4.669 186.805   4.674
  200.25   4.488 207.488   4.581 228.713   4.818 230.347   4.853  250.53   5.582
#Mann= 3 , 0 , 0
  111.46     .04       0 138.226    .033       0 173.022     .03       0
Levee=-1,138.2,3.55,0,,,,
Bank Sta=138.226,173.022
XS Rating Curve= 0 ,0
Exp/Cntr=0.3,0.1

Type RM Length L Ch R = 1 ,814.6489,18.459,18.953,19.95
BEGIN DESCRIPTION:
2008 Survey Section
END DESCRIPTION:
Node Name=BB5
XS GIS Cut Line= 2
299276.9551404685378350.11388619  299099.7180702 5378405.7680387
#Sta/Elev= 15
 106.164    5.82 112.714    5.45 126.584    5.42 136.554    5.73 141.084    3.06
 146.244    1.54 147.014     .87 151.724     .99 166.044    1.61 172.394    1.38
 182.884    4.64 201.784    4.72 221.254    4.36 261.264    5.19 291.934     6.3
#Mann= 3 , 0 , 0
 106.164     .04       0 136.554    .033       0 182.884     .03       0
Levee=-1,136.59,5.75,-1,182.82,4.63,,
#XS Ineff= 2 , 0
       0     140    5.73     179       0     4.6
Permanent Ineff=
       F       F
Bank Sta=136.554,182.884
XS Rating Curve= 0 ,0
Exp/Cntr=0.5,0.3

Type RM Length L Ch R = 3 ,810.68  ,,,
BEGIN DESCRIPTION:
West Street Bridge
END DESCRIPTION:
Bridge Culvert--1,0,-1,-1, 0
Deck Dist Width WeirC Skew NumUp NumDn MinLoCord MaxHiCord MaxSubmerge Is_Ogee
3.97,11.06,1.6,0, 6, 6, , , 0.98, 0, 1,1,,
     125     145     145     175     175     200
    5.43    6.35    6.35    6.35    6.35    4.72
       0       0    4.62    4.62       0       0
  123.09     148     148     178     178   210.5
    5.42    6.35    6.35    6.35    6.35    4.52
       0       0    4.62    4.62       0       0
BR Coef=-1 , 0 , 0 ,, 0 ,,,0.8,-1,,0,
WSPro=,,,, 1 ,,,, 0 ,,,, 0 ,,,,-1 ,-1 ,-1 , 0 , 0 , 0 , 0 , 0
BC Design=,, 0 ,, 0 ,,,,,,
BC Use User HTab Curves=0
BC User HTab FreeFlow(D)= 0

Type RM Length L Ch R = 1 ,795.6959,71.29,57.002,36.886
BEGIN DESCRIPTION:
2008 Survey Section
END DESCRIPTION:
Node Name=BB4
XS GIS Cut Line= 3
299273.9015670265378331.84785611299103.7365074265378384.85630912
299093.8644150325378387.93158407
#Sta/Elev= 17
  104.72    5.39  109.31    3.41  114.22     5.2  115.77    5.34  123.09    5.42
  140.93    5.87   145.7    2.71  151.31    1.45     154     .63  161.41     .64
  163.77    1.07  165.69    1.32  176.53    1.71  184.21     3.6  194.72    4.36
  232.79    4.75  293.29    5.97
#Mann= 3 , 0 , 0
  104.72     .04       0  140.93     .03       0  194.72     .03       0
Levee=-1,140.88,5.86,0,,,,
#XS Ineff= 2 , 0
       0   145.3    5.87     181       0     4.6
Permanent Ineff=
       F       F
Bank Sta=140.93,194.72
XS Rating Curve= 0 ,0
Exp/Cntr=0.5,0.3

Type RM Length L Ch R = 1 ,738.6942,67.074,56.795,41.781
BEGIN DESCRIPTION:
2008 Survey Section
END DESCRIPTION:
Node Name=BB3
XS GIS Cut Line= 3
299199.8787955965378292.15458574299107.6693190495378383.02553655
299098.282487735 5378392.2761073
#Sta/Elev= 13
  187.38    4.09  190.67    4.02  204.99     .82  214.35     .82  220.36    1.82
  221.75    1.06  224.12    2.65  255.08    3.43   283.4    4.45  289.29    2.99
  303.21    2.93  308.78    5.24  330.02    5.95
#Mann= 3 , 0 , 0
  187.38     .04       0  190.67     .03       0  255.08     .03       0
Levee=0,,,-1,283.48,4.45,,
Bank Sta=190.67,255.08
XS Rating Curve= 0 ,0
Exp/Cntr=0.3,0.1

Type RM Length L Ch R = 1 ,681.8989,63.606,55.271,49.993
BEGIN DESCRIPTION:
Interpolated Section
END DESCRIPTION:
Node Name=BB2a
XS GIS Cut Line= 3
299139.2552421285378276.84543925299090.8326266115378398.15095988
299088.4799503045378404.04474776
#Sta/Elev= 23
 241.292   4.024 244.413   3.991 245.096   3.817 247.056   3.149 250.043   2.104
 252.289   1.474 255.851   1.094  258.13     .65 261.649    .404 265.414    .767
 267.017   1.329 267.028   1.329  274.03       3 275.983   3.111  279.49     3.6
  279.86   3.613  281.42   3.983 283.087    3.98 284.582   3.701 308.363   4.271
 334.773   5.056 358.443   5.698 378.251   6.259
#Mann= 3 , 0 , 0
 241.292     .04       0 244.413     .03       0  281.42     .03       0
Levee=0,,,-1,281.4,4.03,,
Bank Sta=244.413,281.42
XS Rating Curve= 0 ,0
Exp/Cntr=0.3,0.1

Type RM Length L Ch R = 1 ,626.6282,58.72,61.011,61.078
BEGIN DESCRIPTION:
2008 Survey Section
END DESCRIPTION:
Node Name=BB2
XS GIS Cut Line= 2
299082.5492337485378262.56919484299085.0328686995378393.97606229
#Sta/Elev= 16
  16.645    3.96  20.175    3.95  23.165    2.67  26.545    1.17  29.085     .35
  33.115     .27  39.675       0  43.175     .46  44.665    1.46  44.675    1.46
  51.185    4.28  56.605    4.54  58.055    5.23  59.605    5.18  60.995    4.59
 148.075    6.56
#Mann= 3 , 0 , 0
  16.645     .04       0  20.175    .033       0  51.185     .03       0
Bank Sta=20.175,51.185
XS Rating Curve= 0 ,0
Exp/Cntr=0.3,0.1

Type RM Length L Ch R = 1 ,565.6174,73.909,74.436,75.815
BEGIN DESCRIPTION:
Interpolated Section
END DESCRIPTION:
Node Name=BB1a
XS GIS Cut Line= 2
299027.9215376945378232.95440991 299015.484348895378365.61775714
#Sta/Elev= 26
  33.236   3.663  42.189   3.724  43.443   3.618  49.773    2.97  55.737    2.34
  58.345   2.022  64.788   1.405   68.87   1.283  70.187    .737  75.009    .754
  77.565    .752  83.028    .604  84.109    .504  91.647    .045  94.064    .313
  95.092    .869  99.593   2.447 103.335   2.613 104.336   2.998 105.406   2.978
 106.366   2.659 110.422   2.758 113.735   3.268 115.193   3.425 149.275   4.147
 166.481   5.015
#Mann= 3 , 0 , 0
  33.236     .04       0  49.773    .033       0  99.593     .03       0
Levee=0,,,-1,104.3,3,,
Bank Sta=49.773,99.593
XS Rating Curve= 0 ,0
Exp/Cntr=0.3,0.1

Type RM Length L Ch R = 1 ,491.1813,180,200,230
BEGIN DESCRIPTION:
2008 Survey Section
END DESCRIPTION:
Node Name=BB1
XS GIS Cut Line= 2
298957.0029866265378194.29174627298946.2925461565378329.32729963
#Sta/Elev= 14
  21.503     3.3  39.253    3.47  60.633    3.21  83.473    2.46  85.763    1.26
  98.593    1.39 108.093    1.17 109.973     .97 123.083      .1 131.583     .36
 133.083    1.36 133.743    1.65 149.173    1.89 156.963    3.13
#Mann= 3 , 0 , 0
  21.503     .04       0  83.473    .033       0 133.743     .03       0
Levee=-1,39.15,3.46,0,,,,
Bank Sta=83.473,133.743
XS Rating Curve= 0 ,0
Exp/Cntr=0.3,0.1

--- Blanche_Brook.g07 (geometry) ---

Geom Title=Base Case - 20% n
Program Version=4.00

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
River Reach=Blanche Brook   ,US of Confluence

Type RM Length L Ch R = 1 ,4158.111,56.608,50.986,38.986
BEGIN DESCRIPTION:
2008 Survey Section
END DESCRIPTION:
Node Name=BB39
XS GIS Cut Line= 2
298673.7152083715380853.34084345 298671.076662985380802.59958592
#Sta/Elev= 12
  36.751   36.56  40.641   36.54  43.971    34.1  50.741   33.98  54.021   33.42
  62.121    33.2  63.911   32.84  64.701   32.62  78.121   32.62  80.281   33.27
  82.021   34.91  87.561   35.35
#Mann= 3 , 0 , 0
  36.751     .08       0  54.021   .0264       0  80.281     .08       0
Bank Sta=54.021,80.281
XS Rating Curve= 0 ,0
Exp/Cntr=0.3,0.1

Type RM Length L Ch R = 1 ,4107.125,48.237,41.636,33.727
BEGIN DESCRIPTION:
Interpolated Section
END DESCRIPTION:
Node Name=BB38a
XS GIS Cut Line= 2
298722.5515181345380829.68306117298690.4697829215380784.29914307
#Sta/Elev= 20
  55.202  35.442  59.493  35.407  63.166  34.288  66.938  34.238  70.459  33.293
  70.634  33.273  74.083  32.656  74.251   32.63  78.273  32.269  83.186  32.159
   85.16  31.975  86.032  31.866  92.064  31.866  93.117  32.273  96.346  32.532
   99.56  33.258  99.796  33.308 106.615  33.442 108.438  34.097  110.78  34.662
#Mann= 3 , 0 , 0
  55.202     .08       0  70.459   .0264       0  99.796     .08       0
Bank Sta=70.459,99.796
XS Rating Curve= 0 ,0
Exp/Cntr=0.3,0.1

Type RM Length L Ch R = 1 ,4065.489,38.598,37.412,37.41
BEGIN DESCRIPTION:
2008 Survey Section
END DESCRIPTION:
Node Name=BB38
XS GIS Cut Line= 2
298755.4837313625380786.51361197 298700.593541525380763.62888025
#Sta/Elev= 14
  58.474   34.53  71.104    34.4  74.894   32.73  78.794   32.01  83.304   31.41
   84.75   31.05    87.5    30.8   90.71   31.04  91.654   31.25  93.134   31.86
 102.184      32 112.094   32.02 114.654   33.15 117.944    34.1
#Mann= 3 , 0 , 0
  58.474     .08       0  74.894    .024       0 114.654     .08       0
Bank Sta=74.894,114.654
XS Rating Curve= 0 ,0
Exp/Cntr=0.3,0.1

Type RM Length L Ch R = 1 ,4028.077,36.768,36.914,37.219
BEGIN DESCRIPTION:
Interpolated Section
END DESCRIPTION:
Node Name=BB37a
XS GIS Cut Line= 2
298751.6701636045380744.77469999298708.0944586265380726.52001277
#Sta/Elev= 19
  55.314  33.941  63.101  33.894  64.351  33.453  65.438  32.889  67.842  32.137
  70.622  31.382  71.835  31.165   73.42   30.88   75.77  30.993  77.278  31.362
  79.355  31.468  84.991  31.485    86.5  31.426  87.672  31.372  96.598  31.403
  97.924  31.691  98.906  32.204  99.206   32.42 102.559  34.573
#Mann= 3 , 0 , 0
  55.314     .08       0  64.351    .024       0  99.206     .08       0
Bank Sta=64.351,99.206
XS Rating Curve= 0 ,0
Exp/Cntr=0.3,0.1

Type RM Length L Ch R = 1 ,3991.163,44.678,43.318,41.969
BEGIN DESCRIPTION:
2008 Survey Section
END DESCRIPTION:
Node Name=BB37
XS GIS Cut Line= 3
298764.9254170855380712.09629316298759.2073460725380709.23725765
298727.7416325775380693.50440091
#Sta/Elev= 14
      62      34  68.393   33.36  71.883    33.4  74.773   30.96  76.293   30.74
    78.3   30.76  79.943   31.05  85.683      31  88.413   30.75    92.5   30.49
   96.05    30.5  98.853    30.8  99.853    31.4 103.573   35.04
#Mann= 3 , 0 , 0
      62     .08       0  71.883    .024       0  99.853     .08       0
Bank Sta=71.883,99.853
XS Rating Curve= 0 ,0
Exp/Cntr=0.3,0.1
